HEC-RAS study SENECACK.prj: SENECACK

--- SENECACK.g03 (geometry) --- (continued)

Type RM Length L Ch R = 1 ,67623   ,399,403.8,394.6
XS GIS Cut Line= 3
2395927.40089043656420.058631069     2396284.579      656282.666
     2396742.406      656077.525
#Sta/Elev= 30
       0 3016.99    72.2 2976.83   127.9 2940.63   192.7 2893.78   247.9 2861.26
   275.9  2841.4   292.9 2828.56   307.9 2814.47   320.7 2791.47   333.6 2775.59
     355 2762.39   363.6 2754.32   398.2  2751.8   405.3 2754.56   414.4 2763.99
   429.6 2765.57   446.4 2775.11   548.4 2818.96   587.6 2839.65   602.1  2849.1
     613 2853.03   648.1 2877.15   687.5 2891.24   700.7 2897.85   709.4 2896.15
   731.3 2881.22     762    2871   805.9 2865.91   854.1 2868.05   884.4 2872.87
#Mann= 4 ,-1 , 0
       0      .1       0   363.6    .045       0   405.3      .1       0
  573.65      .1       0
Bank Sta=363.6,405.3
XS Rating Curve= 0 ,0
Exp/Cntr=0.3,0.1

Type RM Length L Ch R = 1 ,67220   ,350.5,341.8,328.7
XS GIS Cut Line= 3
     2396227.278      656777.8672396418.47753952656577.606112345
     2396968.315      656383.963
#Sta/Elev= 30
       0 2900.55      13 2892.46    37.3 2882.55    59.4 2882.61    86.6 2889.69
   106.4 2891.94   134.7 2886.39   178.8 2872.43   271.5 2832.78   353.5 2790.38
   376.4 2774.02   408.6 2758.48   434.1 2743.03   438.3 2741.11     451 2740.47
   463.8 2742.05   476.5 2748.82   486.2 2764.99   501.9  2785.2   531.6 2814.02
   565.5 2836.66   616.4 2864.43   629.1 2867.54   641.9  2875.7     680 2893.26
     734 2911.23   769.1 2925.93   798.8 2943.52   832.7 2958.97   859.8 2975.06
#Mann= 3 ,-1 , 0
       0      .1       0   434.1    .045       0   463.8      .1       0
Bank Sta=434.1,463.8
XS Rating Curve= 0 ,0
Exp/Cntr=0.3,0.1

Type RM Length L Ch R = 1 ,66878   ,283.9,304.4,326.2
XS GIS Cut Line= 3
      2396415.08      657028.238 2396681.0584355656899.434011101
     2397021.858      656451.605
#Sta/Elev= 30
       0 3042.16    21.8 3025.93    76.5 2993.38   111.5  2969.5   168.5  2936.5
   181.8 2925.21   244.1 2882.27   266.3  2861.1   301.2 2832.52     320 2819.39
   341.4  2798.3   357.8 2784.49   371.3 2768.85   376.6 2764.31   402.7 2747.21
   421.9 2740.31   431.3 2734.98     442 2732.58   465.5 2731.86   479.8 2734.17
   491.2 2738.64   503.1 2753.79     514 2769.96   547.5 2796.21     594 2815.18
   641.8 2839.11   679.6 2862.25   693.9 2867.21   747.5 2896.59   858.3 2962.37
#Mann= 3 ,-1 , 0
       0      .1       0   431.3    .045       0   479.8      .1       0
Bank Sta=431.3,479.8
XS Rating Curve= 0 ,0
Exp/Cntr=0.3,0.1

Type RM Length L Ch R = 1 ,66573   ,297.8,300,298.3
XS GIS Cut Line= 3
2396426.84707212657037.165475726     2396908.459      657023.123
2397317.05233426657030.217072121
#Sta/Elev= 30
       0 3036.56    75.9 2985.75   103.9 2964.96     124  2946.3     140 2939.29
     336 2789.54   368.5 2768.01   416.1 2745.88   436.1 2741.95   448.1 2729.05
   459.12725.854   484.1 2724.15   504.1 2725.62   520.1 2732.85   544.1 2748.66
   552.1 2761.05   560.1 2778.38   568.1 2788.46   600.1 2819.47   628.1 2838.81
   645.1 2858.28   656.1 2873.92   688.3 2892.61   747.3 2931.98   800.2 2972.46
   840.2 3008.47   852.2 3023.31   861.3 3039.75   873.1 3054.92   890.5 3064.18
#Mann= 3 ,-1 , 0
       0      .1       0   459.1    .045       0   504.1      .1       0
Bank Sta=459.1,504.1
XS Rating Curve= 0 ,0
Exp/Cntr=0.3,0.1

Type RM Length L Ch R = 1 ,66273   ,300.2,300,297.1
XS GIS Cut Line= 3
     2396444.269      657350.432      2396850.95       657311.64
     2397264.126      657287.511
#Sta/Elev= 30
       0 3014.52    82.9 2953.09   111.9 2928.37   196.3 2864.17   275.7 2805.47
     328 2768.79     348 2748.96   364.1 2736.18   396.3 2715.27   404.3 2712.74
   420.3 2712.81     428 2715.13   436.4 2720.76   452.4 2725.55   476.4 2750.97
   488.5  2760.8   540.5 2797.68   560.7 2817.36   592.6 2835.87     599 2841.83
   612.7 2859.11   624.5 2865.04   658.6 2871.61   676.8 2878.28   704.8 2876.96
   732.9 2880.15   748.9  2877.6   772.9 2882.15     797 2881.26   822.4 2884.36
#Mann= 3 ,-1 , 0
       0      .1       0   396.3    .045       0     428      .1       0
Bank Sta=396.3,428
XS Rating Curve= 0 ,0
Exp/Cntr=0.3,0.1

Type RM Length L Ch R = 1 ,65973   ,451.2,450,440.1
XS GIS Cut Line= 3
     2396483.807      657676.883     2396892.302       657606.26
2397290.85329681657540.277633844
#Sta/Elev= 30
       0 3016.81    19.2 3002.35   128.8 2906.91   173.5 2873.38   205.9 2843.06
   238.4 2815.56   308.8 2766.65   350.4 2741.46   367.7 2727.46   381.5  2713.1
   396.7 2706.23   416.1 2703.29     430 2706.61   437.3 2715.23   449.5 2716.77
   466.9 2727.48   481.9 2738.71   496.1  2753.8   506.2 2762.13   591.4 2803.28
   619.8 2822.95   656.2 2843.57   664.4 2853.53   692.7 2871.27   708.3 2891.43
     713 2894.61   741.4 2895.82   765.7 2907.08   781.9 2910.78   818.5 2914.66
#Mann= 5 ,-1 , 0
       0      .1       0   396.7    .045       0     430      .1       0
  707.61      .1       0  806.93      .1       0
Bank Sta=396.7,430
XS Rating Curve= 0 ,0
Exp/Cntr=0.3,0.1

Type RM Length L Ch R = 1 ,65523   ,298.3,300,302.4
XS GIS Cut Line= 3
2396619.66755617658206.163149793     2396987.307      658022.978
     2397348.692      657826.846
#Sta/Elev= 30
       0 2967.73    16.7 2966.21    46.5 2949.61    94.2 2921.31   137.5 2892.53
   159.8 2880.16   200.1 2854.35   219.5 2839.41   258.2  2815.4   271.6 2804.36
     312 2776.18   356.5  2739.5   378.8 2712.64   389.5 2704.23   398.5 2694.57
   405.7 2692.41   423.8  2692.8   431.1 2695.18     442 2702.19   454.7 2704.22
   464.7  2716.6   486.4 2730.82   601.3 2795.57   664.1 2840.17   712.8 2871.72
   723.1 2880.63   737.9 2890.44   792.4 2940.84   806.1 2950.02   821.9 2963.85
#Mann= 7 ,-1 , 0
       0      .1       0   65.23      .1       0  273.25      .1       0
   398.5    .045       0   431.1      .1       0  436.66      .1       0
  482.09      .1       0
Bank Sta=398.5,431.1
XS Rating Curve= 0 ,0
Exp/Cntr=0.3,0.1

Type RM Length L Ch R = 1 ,65223   ,299.2,300,301.9
XS GIS Cut Line= 3
     2396766.901      658435.425     2397143.957      658275.604
     2397519.225      658111.714
#Sta/Elev= 30
       0 2838.99    43.3 2822.77    83.4 2801.69     178 2767.29   225.7 2757.72
   247.5 2757.93   277.9 2748.84   303.9 2738.27   321.3 2728.42   338.7 2714.28
   356.1 2706.22   366.4  2698.4   382.1 2696.96   393.9 2689.23   403.9 2686.44
   421.3    2686   433.5  2687.3   436.8 2689.64   456.2 2716.89     479 2739.31
   579.3 2810.15   635.2 2855.65   700.6 2917.75   757.4 2966.33   766.1 2975.97
   774.9 2992.35   779.2 2997.77   796.7 3011.05   805.4 3022.84     819 3032.74
#Mann= 5 ,-1 , 0
       0      .1       0  361.28      .1       0   393.9    .045       0
   436.8      .1       0  463.68      .1       0
Bank Sta=393.9,436.8
XS Rating Curve= 0 ,0
Exp/Cntr=0.3,0.1

Type RM Length L Ch R = 1 ,64923   ,295.3,300,303.9
XS GIS Cut Line= 3
      2396856.26      658697.452     2397241.698      658559.149
     2397627.136      658420.847
#Sta/Elev= 30
       0 2909.01    63.4 2870.99   100.4 2847.02   117.4 2839.85   138.6  2825.3
   232.1 2779.58   304.4 2748.09   342.6 2724.96   363.9 2705.91   372.4 2695.01
   388.6 2684.36   393.6 2681.54   402.1 2680.95   419.9 2681.13   432.4 2684.36
   441.8 2690.39   469.5 2700.64   487.1 2713.36   521.1 2742.76   533.9 2751.73
   548.1 2766.92   587.9 2800.93   606.1 2813.39   665.6 2864.26   682.7 2877.41
   720.8  2911.3   745.2 2930.97   757.7 2943.29   789.3 2969.61     819 2996.68
#Mann= 5 ,-1 , 0
       0      .1       0  369.22      .1       0   388.6    .045       0
   432.4      .1       0   511.9      .1       0
Bank Sta=388.6,432.4
XS Rating Curve= 0 ,0
Exp/Cntr=0.3,0.1

Type RM Length L Ch R = 1 ,64623   ,300,300,298.5
XS GIS Cut Line= 3
     2396922.898      658894.604     2397331.768      658844.394
     2397735.838      658780.636
#Sta/Elev= 30
       0 2904.18    80.4 2847.73   241.6 2751.38   338.4 2698.65   354.5 2686.67
   370.6  2686.7   382.7 2680.34   391.5 2678.87   398.8 2676.57     415 2675.88
   427.1 2676.25   433.3 2678.71   439.3 2683.27   459.5 2711.48   471.4 2723.02
     481 2735.04   508.1 2759.53   524.2 2777.17   548.6 2798.32   560.7 2812.96
   568.8 2819.88   580.2 2835.07   593.1 2847.95   663.7 2903.76   686.3 2918.45
   698.4  2929.8   710.6 2933.96   734.9 2935.83   795.6 2919.54     821  2915.8
#Mann= 3 ,-1 , 0
       0      .1       0   391.5    .045       0   433.3      .1       0
Bank Sta=391.5,433.3
XS Rating Curve= 0 ,0
Exp/Cntr=0.3,0.1

Type RM Length L Ch R = 1 ,64323   ,301.5,300,296.3
XS GIS Cut Line= 3
     2396948.731      659232.003     2397347.392       659140.28
     2397746.101      659036.652
#Sta/Elev= 30
       0 2944.97    30.8 2933.13    59.5 2917.15   121.1 2865.75   182.5 2820.48
   214.4 2794.16   235.8 2781.98   273.1 2753.73   297.6 2740.17   326.3 2720.63
   375.6 2670.56   383.8 2666.88   397.4 2670.86   408.4 2668.94   426.1 2671.41
   442.5 2685.89   453.9 2698.71   478.2 2717.04   507.6 2730.18   536.5 2735.09
   577.9 2730.74   619.2 2719.36   639.3 2720.69   668.8 2718.39     682 2723.23
   734.9 2732.02   751.4 2737.06   763.8 2743.32   780.4 2756.06     821 2777.26
#Mann= 3 ,-1 , 0
       0      .1       0   397.4    .045       0   426.1      .1       0
Bank Sta=397.4,426.1
XS Rating Curve= 0 ,0
Exp/Cntr=0.3,0.1

Type RM Length L Ch R = 1 ,64023   ,307.1,300,289.8
XS GIS Cut Line= 3
2397064.61755319659581.130978735     2397449.602      659418.332
     2397826.983      659249.076
#Sta/Elev= 30
       0 2875.21    32.7 2871.65    58.8 2875.25    71.8 2874.37      98 2864.59
   123.9  2851.4   249.9 2755.15   268.9 2743.71   354.3 2681.23   380.1 2668.52
   397.1  2666.4   406.2 2659.67   406.2 2659.65   410.5 2657.04   419.2 2656.11
   436.2 2659.85   449.9 2661.78   463.8 2675.22   493.8 2699.73   532.7 2716.32
   563.9  2736.1   577.1 2741.61   590.2  2751.2   634.1 2776.36   677.9 2805.23
   751.3 2860.96   787.5 2896.17     805 2907.98   813.8 2917.58   831.6  2933.5
#Mann= 3 ,-1 , 0
       0      .1       0   406.2    .045       0   436.2      .1       0
Bank Sta=406.2,436.2
XS Rating Curve= 0 ,0
Exp/Cntr=0.3,0.1

Type RM Length L Ch R = 1 ,63723   ,444.9,450,451.8
XS GIS Cut Line= 3
2397398.49005799659993.657088958      2397627.17      659647.177
     2397880.284      659317.124
#Sta/Elev= 30
       0 2856.79    13.7 2849.49    29.5 2843.61    60.8 2826.66   109.4 2803.59
   127.9 2796.47   174.7 2774.68   257.3 2738.76   276.5 2732.48   300.5    2719
   324.4 2703.63     358 2677.58   372.4 2661.61   377.1  2658.9   391.5 2656.38
   400.92650.316   427.6 2647.24     435    2650   455.8 2665.11     476 2674.12
   546.6 2714.95   614.7 2761.44   672.6 2798.12   708.9 2827.91   723.2 2837.37
   756.2 2868.44   783.1 2890.86   793.6 2902.03   814.5  2920.4   831.1 2939.18
#Mann= 3 ,-1 , 0
       0      .1       0   400.9    .045       0     435      .1       0
Bank Sta=400.9,435
XS Rating Curve= 0 ,0
Exp/Cntr=0.3,0.1

Type RM Length L Ch R = 1 ,63273   ,434.3,450,461
XS GIS Cut Line= 3
2397670.91702129660198.707872349      2397978.28      659920.882
     2398259.729      659625.401
#Sta/Elev= 30
       0 2762.73    37.5 2746.71     131 2714.18   296.3 2674.04   323.3 2662.52
   359.4 2652.32   369.6 2646.62   382.6 2645.13   392.9 2635.81     415 2632.15
   428.1  2633.5   435.9 2636.43   447.2 2645.04   469.8 2677.16   481.1 2691.04
   499.9 2708.07   555.2 2749.11     560 2754.64     566 2764.65   571.7 2770.45
     589 2780.98   594.8 2790.22   602.8 2798.83   612.2 2812.55   628.2 2827.89
   670.7 2853.27   758.4 2899.49     792  2920.1   800.8 2927.69   822.4 2941.38
#Mann= 5 ,-1 , 0
       0      .1       0   392.9    .045       0   435.9      .1       0
  524.92     .12       0  649.58      .1       0
Bank Sta=392.9,435.9
XS Rating Curve= 0 ,0
Exp/Cntr=0.3,0.1

Type RM Length L Ch R = 1 ,62823   ,448.8,450,450
XS GIS Cut Line= 3
2397720.28848936660409.383680844     2398130.486      660331.679
     2398539.667      660277.388
#Sta/Elev= 30
       0  2805.7    71.7  2773.1    83.9 2768.84   120.5 2751.09   128.7 2749.22
   165.1 2733.67   210.1  2713.4   230.1 2703.14     259 2690.87   267.8 2688.58
   279.3  2682.9   335.8 2662.79   368.9  2645.3   381.1 2634.37   389.3 2632.51
   396.7 2627.25   401.8 2625.51   417.8 2624.16   429.9 2624.92     442 2627.56
   466.2 2646.46   486.1 2653.86   502.5 2661.86   518.6 2674.16   530.7 2679.95
   579.2 2715.88   619.5  2737.5   700.2 2777.87   736.5 2798.14   830.3 2846.35
#Mann= 3 ,-1 , 0
       0      .1       0   396.7    .045       0     442      .1       0
Bank Sta=396.7,442
XS Rating Curve= 0 ,0
Exp/Cntr=0.3,0.1

Type RM Length L Ch R = 1 ,62373   ,303.4,300,298.6
XS GIS Cut Line= 3
2397723.04329787660826.285638313     2398134.535      660778.319
     2398545.138      660725.256
#Sta/Elev= 30
       0 2762.71    23.9 2756.36   172.3 2698.06   258.9 2678.37   285.6 2664.18
   317.8 2641.63   329.9 2636.13     346 2633.91   362.1 2622.26   374.2 2620.91
   388.7  2613.1   410.3 2610.19   430.6 2610.38   435.4 2612.36   442.7 2622.79
   458.9 2638.73     471 2644.21   503.2 2669.94   511.3 2673.84   547.6 2705.16
   575.8 2732.23   628.2 2787.18   660.7 2812.64   672.6 2828.55   684.7 2852.49
   688.8 2857.32   749.3 2897.16   773.5 2905.85   785.5 2916.99   828.3 2932.15
#Mann= 3 ,-1 , 0
       0      .1       0   388.7    .045       0   435.4      .1       0
Bank Sta=388.7,435.4
XS Rating Curve= 0 ,0
Exp/Cntr=0.3,0.1

Type RM Length L Ch R = 1 ,62073   ,302.8,300,295.2
XS GIS Cut Line= 3
     2397820.877      661154.977     2398220.003      661063.387
     2398619.129      660971.797
#Sta/Elev= 30
       0 2802.66   129.1 2725.15   161.9 2708.39     232 2667.78   256.4 2653.06
   268.6 2643.24     281 2637.25   297.4  2624.8     322 2623.82   342.1 2618.69
   383.6 2614.83   393.8 2609.91   404.1 2606.61   436.9 2607.03     441 2609.65
   449.2 2621.01   453.4 2624.76   469.8 2633.54   498.5 2655.98   510.8 2660.54
     519 2666.28     535 2672.28   565.7 2687.88   601.1 2701.68     638 2720.58
   658.6 2728.22   672.6 2731.48   711.9 2734.99   761.2    2735     819 2739.28
#Mann= 3 ,-1 , 0
       0      .1       0   393.8    .045       0     441      .1       0
Bank Sta=393.8,441
XS Rating Curve= 0 ,0
Exp/Cntr=0.3,0.1

Type RM Length L Ch R = 1 ,61773   ,303.1,300,295.3
XS GIS Cut Line= 3
     2397938.852       661504.36     2398316.802      661346.739
     2398694.751      661189.118
#Sta/Elev= 30
       0 2829.13    25.9 2816.61    80.6 2784.22   160.1 2732.89   186.2 2713.58
   196.8 2709.98   259.9 2671.26   298.9 2649.69   311.9 2646.22   372.6 2610.84
   391.1 2606.08   415.9 2602.49   428.9 2602.82   433.3 2605.77   437.6 2611.88
   441.9 2613.96   459.3 2617.34   528.6 2617.52   542.4  2620.7     572 2639.22
   602.3 2667.57   628.3 2688.51   641.3 2701.98   655.5 2712.28   719.3 2749.96
   745.3 2759.37   768.7  2771.9   797.3 2779.53     806 2784.22     819 2795.36
#Mann= 3 ,-1 , 0
       0      .1       0   391.1    .045       0   433.3      .1       0
Bank Sta=391.1,433.3
XS Rating Curve= 0 ,0
Exp/Cntr=0.3,0.1

Type RM Length L Ch R = 1 ,61473   ,287.9,300,314.5
XS GIS Cut Line= 3
     2398123.008      661822.939     2398469.966      661603.128
     2398799.494      661360.385
#Sta/Elev= 30
       0  2753.4     157 2677.87   249.1 2643.99   260.1 2641.89   279.1 2642.55
   307.5 2636.79   331.2 2624.99   359.3 2608.03   376.7 2604.59     388 2598.95
   397.4 2596.61   406.9 2596.31   424.6 2598.91   434.3 2601.62   444.8 2612.34
   454.4  2617.9   476.3 2634.85   491.2 2635.94   501.1 2639.42   545.9 2660.85
   557.4 2667.79   613.5 2709.85   665.1 2751.23   701.1 2783.98   721.4 2800.23
   739.6 2816.66   794.2 2870.98   800.5    2880   809.1 2897.54     820 2908.72
#Mann= 3 ,-1 , 0
       0      .1       0     388    .045       0   424.6      .1       0
Bank Sta=388,424.6
XS Rating Curve= 0 ,0
Exp/Cntr=0.3,0.1

Type RM Length L Ch R = 1 ,61173   ,297.8,300,298.4
XS GIS Cut Line= 3
     2398151.279      661905.618     2398568.819      661878.778
     2398976.547       661865.97
#Sta/Elev= 30
       0  2770.7    67.6 2738.38   155.8 2692.36     228 2659.63     240 2655.62
   308.1 2622.28   324.1 2616.06   348.2 2598.56   376.2 2593.46   384.3 2593.28
   394.9 2590.01   416.3 2589.16   451.2 2590.63   460.3 2591.64   464.4 2593.75
   476.4    2604   492.4 2622.89   501.6 2635.74   524.4 2661.37   544.3 2686.57
   568.4  2711.5   640.4 2742.67   676.5 2762.79   704.5 2780.49   716.5 2792.34
     751 2816.36   780.5 2835.05   792.5 2840.23   812.5  2854.2   826.3 2860.21
#Mann= 5 ,-1 , 0
       0      .1       0   394.9    .045       0   451.2      .1       0
  535.89      .1       0  636.04      .1       0
Bank Sta=394.9,451.2
XS Rating Curve= 0 ,0
Exp/Cntr=0.3,0.1

Type RM Length L Ch R = 1 ,60873   ,300.1,300,298.3
XS GIS Cut Line= 3
2398152.76329787662216.752148916     2398548.024      662173.703
     2398966.084      662132.304
#Sta/Elev= 30
       0  2849.5    42.2 2819.56    78.4 2791.04   142.8 2746.72   163.1 2730.96
   199.2 2706.85   211.2 2696.58   219.3 2692.35   243.4 2673.22   267.6 2657.31
   279.2 2648.07   291.7 2642.65   355.4  2602.1   368.1  2596.8   376.2 2588.19
   384.2 2583.47   396.3 2579.26   415.12583.682   428.5 2585.04   452.6 2605.16
   500.8 2631.76   524.9 2647.32     537 2652.69   669.7 2734.46   697.8 2754.31
   713.9 2761.61   757.4 2795.36   774.2 2805.26   802.3 2829.03   817.7 2835.82
#Mann= 5 ,-1 , 0
       0      .1       0  383.18      .1       0   384.2    .045       0
   415.1      .1       0  482.68      .1       0
Bank Sta=384.2,415.1
XS Rating Curve= 0 ,0
Exp/Cntr=0.3,0.1

Type RM Length L Ch R = 1 ,60573   ,290.6,300,309.6
XS GIS Cut Line= 3
      2398189.35      662523.751     2398596.375      662466.292
2399001.38440426662405.198021285
#Sta/Elev= 30
       0 2742.66    25.6 2737.52   110.5 2724.97   134.7 2718.76   150.7 2713.44
   251.9 2660.61   334.7 2611.99     365 2598.74   373.1 2593.56   381.1 2583.45
   385.2 2579.78   395.7 2575.74   405.1 2573.24   417.5 2572.42   437.7 2574.39
   441.8 2576.81   449.9 2585.48     466 2600.14   482.2 2612.33   490.3 2615.76
   530.8 2644.91   631.9 2706.27   684.5 2741.95   728.9 2773.84   757.1 2795.79
   773.5 2809.99   801.8 2831.27   805.8 2835.05   813.9 2845.45   820.7 2851.93
#Mann= 7 ,-1 , 0
       0      .1       0  197.09      .1       0   395.7    .045       0
   437.7      .1       0  495.09      .1       0  594.41      .1       0
  693.74      .1       0
Bank Sta=395.7,437.7
XS Rating Curve= 0 ,0
Exp/Cntr=0.3,0.1

Type RM Length L Ch R = 1 ,60273   ,302.1,300,293.9
XS GIS Cut Line= 3
     2398171.634      662647.704       2398565.4      662761.001
     2398958.142      662876.537
#Sta/Elev= 30
       0 2684.64      70 2674.21   111.5 2661.79   132.3 2652.89   195.8 2630.55
   257.4 2611.56   325.1 2602.22   344.5 2595.33   361.2 2577.86   373.9  2569.8
   377.8 2567.63   414.8 2566.63   425.2 2568.83   461.2 2584.14   490.4  2603.1
     509 2619.39   528.3  2639.8   548.7 2654.01   573.8 2674.79   589.5 2690.19
     628 2721.08   644.6  2738.9   660.4  2751.6   690.5 2779.17   708.7 2802.56
   723.9 2816.38   757.2 2836.71   794.7 2855.13   807.2 2863.01   819.1 2867.76
#Mann= 9 ,-1 , 0
       0      .1       0  149.34      .1       0  259.16      .1       0
  276.44      .1       0   373.9    .045       0   425.2      .1       0
  478.99      .1       0  735.82      .1       0  809.38      .1       0
Bank Sta=373.9,425.2
XS Rating Curve= 0 ,0
Exp/Cntr=0.3,0.1

Type RM Length L Ch R = 1 ,59973   ,307.4,300,288.7
XS GIS Cut Line= 3
2398059.86485106663037.341872369     2398447.571      663033.014
     2398912.118      663022.418
#Sta/Elev= 30
       0  2773.3   102.9 2708.31   182.9 2664.52   198.9  2653.7   210.9 2650.21
   262.9 2621.09   274.9 2616.11   314.9 2588.75   338.9 2567.22   354.9 2555.12
   368.6 2552.01   394.9 2549.02   402.9 2550.84   405.2 2553.32   414.9 2563.89
   422.9 2569.14   454.9 2577.88   470.7 2585.06   482.9 2593.93   495.3 2598.36
   510.9 2610.98   530.9 2619.88   550.9 2636.82     567 2645.62     611    2679
   694.1 2729.19     715 2739.07     771 2770.83     811 2789.98   852.4 2804.77
#Mann= 5 ,-1 , 0
       0      .1       0   368.6    .045       0   405.2      .1       0
  411.62      .1       0  612.16      .1       0
Bank Sta=368.6,405.2
XS Rating Curve= 0 ,0
Exp/Cntr=0.3,0.1

Type RM Length L Ch R = 1 ,59673   ,291.3,287.8,271
XS GIS Cut Line= 3
2398151.41544677663550.032340402     2398537.764       663313.67
      2398935.74      663103.495
#Sta/Elev= 30
       0 2760.98    55.5 2735.74    65.8 2729.46    78.9 2724.74   132.7  2696.8
   177.4    2678   220.6 2654.53   275.3    2630   318.1 2613.21   330.5 2605.67
   339.3 2603.05   403.3  2555.3   426.6  2552.5     440 2546.06   446.9 2543.49
   467.4 2542.97   482.3 2543.89   488.3 2546.47   494.7 2548.09   512.8 2560.77
   544.5 2560.47   570.2 2565.14   621.5 2589.18   674.8 2619.18   707.3 2641.81
   757.1 2682.83   779.7  2703.8   806.9 2721.68   856.6 2740.25     903 2748.85
#Mann= 5 ,-1 , 0
       0      .1       0     440    .045       0   488.3      .1       0
  536.15      .1       0  640.95      .1       0
Bank Sta=440,488.3
XS Rating Curve= 0 ,0
Exp/Cntr=0.3,0.1

Type RM Length L Ch R = 1 ,59386   ,297.1,312.2,337.4
XS GIS Cut Line= 3
2398468.37802129663821.2983829922398757.72104255663496.875744679
     2398996.764      663166.207
#Sta/Elev= 30
       0 2630.85      43 2640.66    65.7 2639.02   131.9 2617.55   159.8 2603.13
   217.6 2579.25     281 2559.92     332 2554.44   346.1 2546.46   352.1 2545.69
   362.3  2547.2   371.7 2553.82   377.3 2555.15   391.5 2549.31   405.2 2547.03
   414.2 2539.33   428.3 2536.02   466.8 2536.28   474.6 2539.03   491.4 2551.34
     526 2557.77   565.8 2559.36   590.2 2565.19   624.7 2582.85   639.5 2594.23
   649.4 2607.66   654.9 2611.75   717.6 2637.94     753 2656.28   842.7 2690.95
#Mann= 3 ,-1 , 0
       0      .1       0   414.2    .045       0   474.6      .1       0
Bank Sta=414.2,474.6
XS Rating Curve= 0 ,0
Exp/Cntr=0.3,0.1

Type RM Length L Ch R = 1 ,59073   ,295.7,300,301
XS GIS Cut Line= 3
     2398476.596      663854.986     2398887.115      663765.233
     2399286.607      663684.291
#Sta/Elev= 30
       0 2634.64    48.9 2613.38    94.1 2604.72   153.7 2588.62   231.5 2573.55
   247.9  2567.3   288.8 2543.36     297 2542.71   305.2 2545.11   317.5 2541.23
   325.7 2541.27   337.9 2547.44   350.2 2544.95   370.7 2544.82   378.9 2541.73
   391.6 2532.99   407.6 2530.29   432.1 2531.03   444.3 2533.83   456.6 2550.06
   464.7 2563.19   472.9 2571.68   481.1    2583   513.5 2616.51     530 2632.23
   615.7 2697.97   623.9  2700.6   653.6 2721.31   701.4 2750.46   827.8 2811.91
#Mann= 3 ,-1 , 0
       0      .1       0   391.6    .045       0   444.3      .1       0
Bank Sta=391.6,444.3
XS Rating Curve= 0 ,0
Exp/Cntr=0.3,0.1

Type RM Length L Ch R = 1 ,58773   ,311.3,300,289.4
XS GIS Cut Line= 3
     2398477.073      664098.781     2398884.169      664064.714
     2399295.589      664009.886
#Sta/Elev= 30
       0 2730.08    33.8 2716.84    45.8  2707.6   123.7 2656.26   142.1 2642.04
   190.5 2610.52   234.8 2585.05   247.3  2579.5   306.7 2541.42   342.9  2535.1
   358.9 2533.92     375 2529.31     383 2529.25     383 2529.26   399.1 2525.74
   411.1 2525.41   423.4 2525.62   435.3 2528.25   447.4 2536.34   491.8 2536.28
   503.9 2539.09   515.7 2543.58   524.1 2547.96   536.2 2562.19   572.7 2581.81
   584.6 2595.07   592.7 2600.46   673.4 2621.18   790.4 2656.94   823.6 2669.46
#Mann= 3 ,-1 , 0
       0      .1       0     383    .045       0   435.3      .1       0
Bank Sta=383,435.3
XS Rating Curve= 0 ,0
Exp/Cntr=0.3,0.1

Type RM Length L Ch R = 1 ,58473   ,289.6,300,307.8
XS GIS Cut Line= 3
     2398609.112        664533.8     2398968.978      664346.212
2399371.96320332664143.026539023
#Sta/Elev= 30
       0 2689.43    33.4 2683.58    96.6 2681.94   123.6 2679.09   153.4 2671.96
   173.3 2665.53   181.3 2661.22   279.7 2590.78   304.1 2570.16   317.7 2560.83
   326.6 2552.45   335.5 2547.44   353.7 2530.42   371.7  2522.9   380.8  2520.9
   412.6 2520.49   433.4 2520.83   439.2 2523.07   448.1 2528.74   452.6 2529.48
   504.9 2529.14   537.6 2526.13   582.5 2528.81   600.4 2536.94   649.7    2566
   667.6 2573.94   721.4  2592.9   788.6 2619.41   815.5 2630.93   857.1 2653.21
#Mann= 5 ,-1 , 0
       0      .1       0   371.7    .045       0   439.2      .1       0
  527.93      .1       0  632.09      .1       0
#XS Ineff= 2 , 0
                          483.92         2534.96
Permanent Ineff=
       F       F
Bank Sta=371.7,439.2
XS Rating Curve= 0 ,0
Exp/Cntr=0.3,0.1

Type RM Length L Ch R = 1 ,58173   ,277,302.1,324.9
XS GIS Cut Line= 3
      2398647.53       664594.77     2399191.081      664533.225
       2399575.3      664505.328
#Sta/Elev= 30
       0  2648.5    79.7 2624.63    99.1 2621.06   152.2 2604.37   241.5 2572.51
   256.8 2565.66   293.1 2554.57   342.7 2533.88   357.5 2529.44   369.6 2522.74
   381.6 2522.36   409.8 2529.72   478.3 2521.34   490.3  2518.2   506.4 2518.33
   521.3 2516.08   530.6 2514.06   554.7 2513.18   570.8 2513.69   578.8 2515.81
   578.8 2515.82   598.8 2524.44   614.9 2537.53   638.9 2550.17     683 2561.37
   715.1 2578.35   723.2 2580.15   759.2 2595.05   839.5  2598.7   932.3 2605.92
#Mann= 5 ,-1 , 0
       0      .1       0  474.06      .1       0   521.3    .045       0
   578.8      .1       0  772.97      .1       0
Bank Sta=521.3,578.8
XS Rating Curve= 0 ,0
Exp/Cntr=0.3,0.1

Type RM Length L Ch R = 1 ,57871   ,297.6,297.9,295.2
XS GIS Cut Line= 3
     2398623.371      664664.0152398913.59365464664661.915545071
     2399346.618      665048.455
#Sta/Elev= 30
       0 2630.13    31.4  2616.5    47.4 2613.38    66.7 2604.88   131.4 2584.06
   147.4 2575.66   223.4 2545.36     236 2542.49   260.1 2528.89   279.4 2521.33
   354.1 2520.52   372.2 2515.39   388.3 2522.35   425.8 2506.82   474.1 2505.16
   490.2 2506.93   529.7 2513.23   570.6 2538.78     586 2557.07     598 2567.58
     651 2606.21   677.8 2629.16   683.2 2635.65   694.1 2655.69   719.5 2676.61
   736.8 2697.58   758.3 2718.22   804.5 2734.03   832.3 2746.92   870.7 2749.67
#Mann= 4 ,-1 , 0
       0      .1       0   425.8    .045       0   490.2      .1       0
  747.05      .1       0
Bank Sta=425.8,490.2
XS Rating Curve= 0 ,0
Exp/Cntr=0.3,0.1

Type RM Length L Ch R = 1 ,57573   ,306.3,300,295.4
XS GIS Cut Line= 3
     2398569.045      664757.155     2398880.358      665024.844
     2399200.449      665279.944
#Sta/Elev= 30
       0 2615.41     7.5 2610.74    16.6 2608.61    49.7 2588.96   110.2 2565.93
   134.1 2559.35   161.3 2547.36   218.5 2509.93   260.7  2505.8   334.6 2506.11
   354.2 2501.45   362.7 2497.06   368.3 2491.62   376.8 2487.88   397.9 2487.66
   416.6 2488.07   425.1 2491.34   439.3 2498.97   452.4 2501.63     475 2501.66
     482 2504.41   504.8 2518.55   551.7 2555.29   621.5 2599.67   633.6 2611.18
   664.6 2627.21   696.3 2637.92   743.9 2648.78   780.9 2652.49   819.9 2653.62
#Mann= 4 ,-1 , 0
       0      .1       0   368.3    .045       0   425.1      .1       0
  674.85      .1       0
Bank Sta=368.3,425.1
XS Rating Curve= 0 ,0
Exp/Cntr=0.3,0.1

Type RM Length L Ch R = 1 ,57273   ,308.2,300,291.9
XS GIS Cut Line= 3
     2398321.581       665042.32     2398678.993      665242.064
     2399029.121      665455.088
#Sta/Elev= 30
       0 2645.07    25.8 2635.61    51.2 2618.74   111.3 2593.27   134.2 2580.33
   225.9 2572.76   244.2 2567.09   267.1  2553.8   285.4 2537.05   329.1 2504.51
   362.8 2494.09   371.7 2485.88   378.3 2484.01   426.4 2483.74   434.1 2485.88
   441.9  2487.6     470 2486.89   488.5 2492.96   508.8 2492.73   526.2 2495.69
   568.3 2493.21   601.1 2493.67   619.5 2496.52   634.2 2500.21   671.4 2522.08
   703.5 2534.45   715.5  2536.1   736.9 2543.36   783.7 2553.52   819.3 2558.46
#Mann= 5 ,-1 , 0
       0      .1       0  268.62    .055       0  345.82      .1       0
   371.7    .045       0   434.1      .1       0
Bank Sta=371.7,434.1
XS Rating Curve= 0 ,0
Exp/Cntr=0.3,0.1

Type RM Length L Ch R = 1 ,56973   ,285.5,300,314.4
XS GIS Cut Line= 3
     2398182.528      665415.969     2398579.646      665520.683
2398971.02066574665627.000224689
#Sta/Elev= 30
       0 2690.23    38.6 2666.77   157.4 2602.78   169.8 2593.23   178.1 2589.75
   202.9 2568.48   219.5 2568.97   227.7  2566.1   252.6 2548.06     271 2529.57
   288.3 2516.23   298.1 2511.83   322.9 2505.95   347.7 2491.08   359.4 2490.14
   372.5 2483.02   388.8 2478.67   405.6 2475.85   447.6  2478.3   471.9 2481.52
   513.4 2483.14   538.9 2487.13   556.4 2492.82   596.3 2490.67     617 2493.11
   663.2 2494.73   679.2 2498.26   695.8 2497.81   757.9 2504.85   816.2 2518.86
#Mann= 5 ,-1 , 0
       0      .1       0  186.17    .055       0  294.87      .1       0
   388.8    .045       0   447.6      .1       0
Bank Sta=388.8,447.6
XS Rating Curve= 0 ,0
Exp/Cntr=0.3,0.1

Type RM Length L Ch R = 1 ,56673   ,310.4,300,293.3
XS GIS Cut Line= 3
     2398135.265      665497.428     2398435.227      665775.786
2398739.78385021666061.066002775
#Sta/Elev= 30
       0  2705.7    13.9 2695.77   167.7 2598.63     196 2577.68   213.8  2560.2
   218.6 2557.92   232.8 2557.46   237.4 2556.22   255.4 2543.71   269.6  2535.8
   288.5 2519.26   326.2 2491.83   337.3 2481.36     355 2474.71   370.4 2462.44
   377.1 2460.49   399.8 2459.32     425 2459.81   431.3 2461.84   437.2 2466.67
   454.7 2472.13   472.3 2480.65   501.7 2478.75   523.7 2483.06   534.6 2483.79
   612.7  2481.4   649.7 2476.93   704.5 2481.56   803.2 2474.23   826.5 2474.76
#Mann= 3 ,-1 , 0
       0      .1       0   370.4    .045       0   431.3      .1       0
Bank Sta=370.4,431.3
XS Rating Curve= 0 ,0
Exp/Cntr=0.3,0.1

Type RM Length L Ch R = 1 ,56373   ,308,300,292.6
XS GIS Cut Line= 3
     2397924.812      665851.567     2398289.766      666037.303
     2398655.663      666221.192
#Sta/Elev= 30
       0 2657.71    42.6 2632.63    72.3 2612.33    86.7  2607.7   105.4 2593.28
   161.6 2561.26   181.7 2545.62   208.6 2542.61     267 2497.12   289.4 2482.05
   301.4 2478.45   328.1 2479.57     346 2469.17   365.7  2468.1   379.2 2456.67
   383.7 2454.56   405.5 2454.07   430.9 2454.59   437.5  2457.2   446.4 2461.13
   509.7 2460.17   518.7 2463.18   535.9 2474.52   546.7 2475.65   578.3 2475.45
   607.6  2470.7   655.7  2471.4   674.7 2474.59   791.1 2469.34     819 2469.88
#Mann= 3 ,-1 , 0
       0      .1       0   379.2    .045       0   437.5      .1       0
#XS Ineff= 2 , 0
                          469.03         2468.11
Permanent Ineff=
       F       F
Bank Sta=379.2,437.5
XS Rating Curve= 0 ,0
Exp/Cntr=0.3,0.1

Type RM Length L Ch R = 1 ,56073   ,281.6,300,307.6
XS GIS Cut Line= 3
2397817.14070319666247.334080447     2398215.126      666324.384
     2398613.675      666410.824
#Sta/Elev= 30
       0 2535.71    13.9 2529.47    26.1 2521.53    50.5 2521.18    66.8  2512.7
    89.7 2505.37   197.2 2485.43   209.2 2480.22   243.3 2460.13     257 2456.02
   266.5 2448.77   274.1  2447.5   323.5 2451.98   372.4 2450.91   412.1 2448.81
   425.5 2451.36   462.3 2458.69   507.3  2455.5   528.2 2464.48     536 2465.98
   568.9  2464.3   597.4 2466.24   621.9  2463.9     646 2466.73   691.5 2464.84
     712 2467.88   769.3 2467.71   785.6    2466   797.9 2468.05   813.2 2475.75
#Mann= 3 ,-1 , 0
       0      .1       0   372.4    .045       0   425.5      .1       0
Bank Sta=372.4,425.5
XS Rating Curve= 0 ,0
Exp/Cntr=0.3,0.1

Type RM Length L Ch R = 1 ,55773   ,311.9,300,298.8
XS GIS Cut Line= 3
      2397729.42      666302.964      2398048.23      666553.501
     2398390.057      666818.177
#Sta/Elev= 30
       0 2542.47    57.9 2514.12    69.3 2506.48    93.3 2505.36   103.4 2499.88
   129.1 2492.83     195 2479.81     251  2470.4   257.3 2467.36   277.2 2453.17
   286.6 2451.55   297.7 2447.63   325.6 2447.29   337.4 2445.33   362.9 2443.71
   374.1 2441.41   391.2 2440.77   411.1 2441.36   420.8 2443.27   442.5 2446.01
   454.2 2450.43   489.6 2453.65     558 2449.67     605 2449.73   646.4 2446.18
   695.2 2448.57     719 2451.07   732.4 2457.58     741 2463.98   837.8 2547.54
#Mann= 3 ,-1 , 0
       0      .1       0   362.9    .045       0   420.8      .1       0
#XS Ineff= 2 , 0
                          491.79         2462.66
Permanent Ineff=
       F       F
Bank Sta=362.9,420.8
XS Rating Curve= 0 ,0
Exp/Cntr=0.3,0.1

Type RM Length L Ch R = 1 ,55473   ,276.9,300,309.5
XS GIS Cut Line= 3
     2397572.045       666648.77     2397949.551      666833.302
2398279.10025381666992.897077672
#Sta/Elev= 30
       0 2479.68    16.4 2477.23    83.1 2477.79   108.3 2472.65   141.2 2470.99
     186 2445.54     195 2442.46   225.6 2444.12     239 2441.33   251.8 2442.18
     288 2438.61   323.6    2439   336.9 2435.62   363.6 2440.25   396.5 2438.93
   408.2 2435.47     426 2434.71   443.7 2435.04   449.2 2437.66   461.5 2447.73
   488.2 2449.56   521.1 2447.81     546 2449.95   613.9 2449.97   652.8 2442.34
     666 2443.28   688.8 2455.89   742.7 2501.59   775.6 2535.58   786.4 2553.35
#Mann= 3 ,-1 , 0
       0      .1       0   396.5    .045       0   449.2      .1       0
#XS Ineff= 2 , 0
                           592.2         2461.89
Permanent Ineff=
       F       F
Bank Sta=396.5,449.2
XS Rating Curve= 0 ,0
Exp/Cntr=0.3,0.1

Type RM Length L Ch R = 1 ,55173   ,284.7,300,301.4
XS GIS Cut Line= 3
     2397528.708      666719.161     2397825.718      667098.757
     2398035.192      667435.652
#Sta/Elev= 30
       0  2473.7    61.7  2462.9   106.3 2462.05   140.9 2441.87   146.9 2439.71
   172.1 2441.32   217.5 2438.23   230.5  2439.5   257.7  2438.9     289 2433.86
   304.4 2437.21   317.5 2436.88   323.2 2435.71   329.8 2432.09   351.7 2429.99
     411 2436.08   434.4 2433.02   477.1 2431.56     501 2432.99     509 2435.78
     534 2433.23   567.1 2434.81   607.7 2431.98   619.3 2432.85   662.9 2468.61
   703.5 2506.11   717.6 2516.38   753.2 2535.59   835.4 2586.81   878.7 2610.57
#Mann= 3 ,-1 , 0
       0      .1       0   434.4    .045       0     501      .1       0
#XS Ineff= 2 , 0
          409.57 2448.11  507.14         2446.82
Permanent Ineff=
       F       F
Bank Sta=434.4,501
XS Rating Curve= 0 ,0
Exp/Cntr=0.3,0.1

Type RM Length L Ch R = 1 ,54873   ,347,321,307.6
XS GIS Cut Line= 3
     2397369.804       666792.11      2397542.16      667151.235
2397745.21510637667556.972808514
#Sta/Elev= 30
       0 2490.04   140.7 2468.34   152.7 2464.83   171.7 2456.81   196.3 2442.39
   214.8 2436.59   242.5 2433.47     327 2434.75   344.6 2430.64   353.5 2426.53
   380.5 2424.39   414.2 2425.94   456.1 2423.82   465.1  2424.8     485 2430.05
   514.3 2427.61   529.7 2428.26   569.5 2426.68   598.3 2422.15   661.9 2426.03
   693.2 2425.08   697.6 2425.55   715.5 2432.47   724.5 2437.86   748.2 2458.28
   755.8  2465.9   772.3 2486.98   782.6 2497.67   809.9 2518.49   852.1 2546.96
#Mann= 3 ,-1 , 0
       0      .1       0   353.5    .045       0   414.2      .1       0
#XS Ineff= 2 , 0
                          485.38         2435.49
Permanent Ineff=
       F       F
Bank Sta=353.5,414.2
XS Rating Curve= 0 ,0
Exp/Cntr=0.3,0.1

Type RM Length L Ch R = 1 ,54552   ,273.5,279,277.8
XS GIS Cut Line= 3
      2396970.34      667255.6222397222.61785102667340.737872329
2397711.80772339667563.748765944
#Sta/Elev= 30
       0 2494.33     106  2477.9   139.7 2475.32   165.1 2471.38     186 2464.31
   223.9 2446.25   245.3 2433.87   261.7 2428.78   349.9  2425.8   363.1 2424.23
   370.6 2420.33   407.1 2418.62   424.6 2420.53   443.1 2419.33   455.2 2420.69
   470.3 2416.87   500.5 2417.52     517  2422.1   547.7 2418.91   604.9 2421.69
   615.2 2424.24   626.9 2422.14   648.4 2425.19   679.6 2426.49   692.8 2433.34
   719.2 2454.88   723.6 2459.36   736.8 2479.53   754.1 2496.25   803.9 2530.95
#Mann= 3 ,-1 , 0
       0      .1       0   370.6    .045       0   424.6      .1       0
Bank Sta=370.6,424.6
XS Rating Curve= 0 ,0
Exp/Cntr=0.3,0.1

Type RM Length L Ch R = 1 ,54273   ,284.2,300,297.5
XS GIS Cut Line= 3
     2396913.667       667435.26     2397311.552      667669.864
2397670.86459574667866.476574478
#Sta/Elev= 30
       0 2468.16    52.3 2460.29   140.6 2442.75   169.9 2433.37   190.4 2421.75
   199.2 2422.02   210.8 2426.52   225.4 2421.23   275.2 2418.18   326.3 2420.91
   348.1 2414.69   372.7 2413.37   419.2 2415.32   428.5 2414.36   450.4 2412.14
   474.7 2411.86   479.7 2414.01   485.6 2417.83     514  2419.2   529.4 2418.41
   541.6 2414.53   559.3 2412.92   572.4 2414.46   588.7 2426.73   606.9 2447.36
   643.4 2482.18   679.8 2510.78     798  2588.9   839.4 2613.77   871.5 2631.03
#Mann= 3 ,-1 , 0
       0      .1       0   428.5    .045       0   479.7      .1       0
#XS Ineff= 2 , 0
                          508.21         2440.72
Permanent Ineff=
       F       F
Bank Sta=428.5,479.7
XS Rating Curve= 0 ,0
Exp/Cntr=0.3,0.1

Type RM Length L Ch R = 1 ,53973   ,306.7,300,282.2
XS GIS Cut Line= 3
     2396805.205      667536.921     2397079.261      667829.203
     2397418.768      668138.432
#Sta/Elev= 30
       0 2459.89   123.3 2437.18   136.8 2432.59   161.7 2420.27   171.8 2417.32
   206.2 2419.42   237.4 2417.63   248.7 2415.93   262.8  2410.7   288.3 2407.93
   319.4 2411.47   347.3 2409.46   376.5 2411.12   384.5 2408.46   405.4 2406.43
   432.6 2408.67   448.7  2409.8   472.3 2407.12   481.1 2409.27   526.1 2411.49
   556.9 2405.63   569.5  2407.3   581.4 2415.67     611 2446.71   633.7  2473.1
   646.7 2484.62     713 2529.32   778.7 2579.83   812.1 2601.05   859.9 2628.48
#Mann= 3 ,-1 , 0
       0      .1       0   384.5    .045       0   432.6      .1       0
Bank Sta=384.5,432.6
XS Rating Curve= 0 ,0
Exp/Cntr=0.3,0.1

Type RM Length L Ch R = 1 ,53673   ,293.2,300,315.6
XS GIS Cut Line= 3
     2396578.535      667957.418     2396989.062      668098.962
     2397381.505      668212.373
#Sta/Elev= 30
       0 2406.02    17.1 2403.59      51 2407.29   105.2 2407.76   135.6 2405.65
   177.9 2409.77   199.5 2402.65   228.7 2404.25   240.4 2400.39   254.1 2399.28
   279.5 2401.83   334.5 2402.86     360 2399.99   410.6 2403.87   421.8 2401.04
   456.8 2399.16   469.3 2400.66   477.5 2403.44   487.2 2400.24   503.4 2400.42
   515.1 2404.72   522.8 2411.24   548.1 2448.92   556.7 2464.62   565.6 2474.43
   610.9 2506.83     715 2576.21   819.9 2638.71   836.1 2643.61   842.7 2647.96
#Mann= 3 ,-1 , 0
       0      .1       0   421.8    .045       0   469.3      .1       0
#XS Ineff= 2 , 0
           221.6 2442.05
Permanent Ineff=
       F       F
Bank Sta=421.8,469.3
XS Rating Curve= 0 ,0
Exp/Cntr=0.3,0.1

Type RM Length L Ch R = 1 ,53373   ,151.7,150,150.1
XS GIS Cut Line= 3
     2396514.236      668040.742     2396807.038      668327.024
      2397099.84      668613.305
#Sta/Elev= 30
       0 2405.31    23.1 2402.94    39.9  2403.7    71.7 2401.68    98.1 2398.87
   171.6 2400.05   190.9 2398.08   231.9 2398.22     314 2401.76   319.6 2401.32
   330.8 2395.67   336.4 2394.21   364.3 2392.34   383.7 2392.94   423.3 2393.53
   426.2 2395.25   437.9 2421.39   448.2 2436.04   453.8  2442.4   466.5 2453.55
   489.4 2470.44   537.8 2500.42   576.9 2527.13   652.5 2571.37   701.1 2610.45
   714.7 2615.12   740.1 2630.01   752.6 2631.36   771.3  2640.2     819 2670.12
#Mann= 3 ,-1 , 0
       0      .1       0   383.7    .045       0   423.3      .1       0
#XS Ineff= 2 , 0
          292.61 2428.88
Permanent Ineff=
       F       F
Bank Sta=383.7,423.3
XS Rating Curve= 0 ,0
Exp/Cntr=0.3,0.1

Type RM Length L Ch R = 1 ,53223   ,289.2,300,307.1
XS GIS Cut Line= 3
     2396409.371      668147.996     2396702.173      668434.277
     2396994.975      668720.559
#Sta/Elev= 30
       0 2403.45     7.5 2401.49    32.7 2400.03    67.1 2401.25      97  2396.1
   124.3 2396.29     136 2394.27   175.3 2395.24     193  2392.6   215.8 2393.96
   242.5 2399.52   266.1 2399.97   273.1 2399.08   290.2 2391.56   348.1 2393.46
   362.3 2390.49   410.3 2389.94   418.8 2391.29   424.5 2395.48   471.8 2444.86
   501.9 2470.68   526.3 2489.13   604.9 2540.28     645 2564.34   662.1 2577.02
   676.2 2582.09   751.5 2640.59   763.9 2644.46   775.2 2653.71     819 2678.15
#Mann= 3 ,-1 , 0
       0      .1       0   362.3    .045       0   418.8      .1       0
#XS Ineff= 2 , 0
          262.54  2411.4
Permanent Ineff=
       F       F
Bank Sta=362.3,418.8
XS Rating Curve= 0 ,0
Exp/Cntr=0.3,0.1

Type RM Length L Ch R = 1 ,52923   ,302.7,300,296.3
XS GIS Cut Line= 3
     2396291.009      668248.866     2396468.882      668617.851
     2396638.563      668990.519
#Sta/Elev= 30
       0 2436.83    49.3 2404.91    63.9 2398.22    73.3 2395.75   148.8 2393.66
     171 2390.35   188.7 2389.66     202 2386.69   237.6 2385.88   370.8 2387.45
   384.8 2384.45     393 2382.14   406.3 2381.88   417.9 2382.22   432.7 2384.53
   462.4    2385   469.2 2386.94   487.3 2388.41   494.3 2390.11   512.9  2397.7
   520.6 2401.74     530 2408.53   558.9 2435.19   577.9 2449.63   602.1 2463.96
   630.5 2482.49   648.1 2491.93   661.3 2503.28   771.2 2557.38   819.1 2583.94
#Mann= 3 ,-1 , 0
       0      .1       0   384.8    .045       0   432.7      .1       0
Bank Sta=384.8,432.7
XS Rating Curve= 0 ,0
Exp/Cntr=0.3,0.1

Type RM Length L Ch R = 1 ,52623   ,322.6,300,283.7
XS GIS Cut Line= 3
     2396003.055      668360.572     2396187.999      668718.739
 2396409.9222825669099.365332265
#Sta/Elev= 30
       0 2449.41    52.1 2440.21    63.8 2439.95   133.2 2429.77   151.2  2423.1
   191.1 2398.41   206.3  2390.9   214.2 2388.69   313.2 2384.72   330.6  2386.3
   348.1 2385.73   365.5 2377.91   374.2 2376.07   407.9 2375.74   431.1 2377.67
   444.9 2376.32   469.6 2379.63   487.1 2379.16   501.7 2382.94   577.8 2380.05
   616.3 2380.74   630.9 2377.98   653.8 2380.61     686 2378.75   703.6 2381.97
     727 2390.68   750.4 2405.31   801.5 2448.13   821.5 2462.08   843.7  2475.1
#Mann= 3 ,-1 , 0
       0      .1       0   365.5    .045       0   431.1      .1       0
#XS Ineff= 2 , 0
                          513.13         2390.85
Permanent Ineff=
       F       F
Bank Sta=365.5,431.1
XS Rating Curve= 0 ,0
Exp/Cntr=0.3,0.1

Type RM Length L Ch R = 1 ,52323   ,298.2,300,300.3
XS GIS Cut Line= 3
     2395677.799      668794.286     2396047.169      668973.247
     2396403.891      669174.005
#Sta/Elev= 30
       0 2458.32    63.3 2452.85    89.9 2447.77   114.9 2439.66   134.4 2429.11
   183.8 2391.56   201.1 2383.92   227.7  2377.3   276.6 2377.75   300.6 2374.77
   347.7 2377.57   384.4 2372.87   392.2 2369.33   405.4 2368.87   432.9 2369.18
   443.6 2372.73   452.5 2378.07   469.6 2379.08     488  2376.9   552.2 2377.78
     566 2374.61   593.6 2376.83   616.9 2370.98   675.7 2377.13   699.2 2391.89
   722.7 2414.32   743.2 2438.85   760.8 2454.13   796.1 2478.93   819.8 2500.99
#Mann= 3 ,-1 , 0
       0      .1       0   384.4    .045       0   443.6      .1       0
#XS Ineff= 2 , 0
          340.57    2384  508.91         2384.93
Permanent Ineff=
       F       F
Bank Sta=384.4,443.6
XS Rating Curve= 0 ,0
Exp/Cntr=0.3,0.1

Type RM Length L Ch R = 1 ,52023   ,296.7,300,303.3
XS GIS Cut Line= 3
     2395543.987      669030.041     2395899.017      669234.109
     2396254.047      669438.178
#Sta/Elev= 30
       0 2452.23    40.1 2438.75    49.5 2434.45    63.2 2431.34    95.5 2410.63
   134.5 2383.02   155.4    2371     160 2369.55   348.3  2371.4     363 2368.59
   374.7 2369.24   381.5 2366.49   390.7 2364.31   427.5 2364.69   439.2 2367.38
   464.6 2370.55   510.7 2372.54   609.1 2373.82   658.9 2372.73   667.6 2371.21
   682.3 2365.36   704.5 2364.64   709.1 2365.99   713.7 2369.15   732.2 2384.57
   743.9 2395.75   758.5 2412.62   767.3 2420.31   811.2 2446.78     819 2450.26
#Mann= 3 ,-1 , 0
       0      .1       0   381.5    .045       0   439.2      .1       0
#XS Ineff= 2 , 0
           319.3 2380.39  523.61         2380.82
Permanent Ineff=
       F       F
Bank Sta=381.5,439.2
XS Rating Curve= 0 ,0
Exp/Cntr=0.3,0.1

Type RM Length L Ch R = 1 ,51723   ,304.7,300,296.2
XS GIS Cut Line= 3
     2395408.047      669247.026     2395739.395      669487.647
     2396070.743      669728.269
#Sta/Elev= 30
       0 2455.18    20.2 2444.19    79.2 2417.16   146.7 2397.61     211 2386.17
   255.4 2363.09   282.5 2361.41   299.7 2362.84   319.7 2360.62   351.2 2364.18
   368.4 2364.11     377 2362.43   387.8 2359.38   433.4 2359.28   438.4  2360.5
   442.2 2363.44   448.6 2366.15   508.7 2362.67   531.6 2366.42   600.4 2367.21
   631.2 2361.12   689.1 2365.77   700.4 2362.55   712.1 2364.75   725.1 2358.99
   741.8 2357.96   749.8 2359.11   779.5 2371.19   794.3 2382.65     819 2405.09
#Mann= 5 ,-1 , 0
       0      .1       0  371.81      .1       0     377    .045       0
   442.2      .1       0  487.94      .1       0
Bank Sta=377,442.2
XS Rating Curve= 0 ,0
Exp/Cntr=0.3,0.1

Type RM Length L Ch R = 1 ,51423   ,270.3,256.8,245.3
XS GIS Cut Line= 3
     2395203.035      669537.685     2395563.073      669730.225
2395994.42604168669947.284650202
#Sta/Elev= 30
       0 2490.41   148.5 2415.91   167.5 2401.87   181.1 2389.13   208.3 2367.11
   222.3 2358.25   249.2 2356.12   367.1 2358.13   373.1 2356.47     379 2354.51
   394.3 2354.21   421.4 2354.38   432.4 2356.65   439.3 2359.15   456.2 2359.36
     489 2355.73   510.9 2358.34   554.5 2356.85   590.3 2357.98   627.3 2353.99
   654.2 2357.63   672.1 2356.47     690 2357.88   742.2  2355.5   761.7  2359.2
   834.5 2360.73   842.3 2363.35   852.4 2369.73   882.6 2394.22   891.2 2403.38
#Mann= 5 ,-1 , 0
       0      .1       0   370.8      .1       0   373.1    .045       0
   432.4      .1       0  500.18      .1       0
Bank Sta=373.1,432.4
XS Rating Curve= 0 ,0
Exp/Cntr=0.3,0.1

Type RM Length L Ch R = 1 ,51167   ,201.3,193.2,184.1
XS GIS Cut Line= 3
     2395065.902      669917.151 2395198.1876918669947.476282502
     2395910.357      669998.633
#Sta/Elev= 30
       0 2503.14    58.3 2471.12      87 2457.14   103.5 2450.53   172.4 2416.38
     233 2391.57   252.6 2378.49   256.6 2373.12   264.6 2358.89   268.6 2354.86
   276.6 2350.51   284.7 2348.76   304.7 2350.99   320.7 2349.96   356.8 2353.81
   372.9 2350.96   380.9 2349.31     435 2351.14   453.1 2352.06   469.1 2350.72
   481.2 2351.55   501.2 2349.45   541.3 2349.98   562.2 2353.15   597.5 2352.34
   696.9 2353.35   711.9 2355.04   733.8 2354.77   749.3 2357.14   849.7 2359.14
#Mann= 3 ,-1 , 0
       0      .1       0   372.9    .045       0     435      .1       0
Bank Sta=372.9,435
XS Rating Curve= 0 ,0
Exp/Cntr=0.3,0.1

Type RM Length L Ch R = 1 ,50973   ,328.2,331.3,336.3
XS GIS Cut Line= 3
     2395084.566      670249.455     2395474.552      670154.666
     2395915.758      670040.512
#Sta/Elev= 30
       0  2434.5    35.2    2428   103.3 2418.38   146.3 2408.56   202.6 2387.84
   236.9 2372.34   282.1  2348.4     311 2346.69   323.3 2343.98   335.7 2345.83
     345 2345.06   368.2 2349.13   374.7 2348.23   389.2 2346.08   409.8 2345.88
   424.3 2347.39   476.8 2347.78   517.2  2346.1   552.4 2349.12   608.1 2349.84
   632.9 2354.59   670.1 2353.56   680.3 2349.78   686.6 2349.31   711.4 2353.97
   765.1 2356.91   777.5 2355.88   831.3 2356.32   843.6 2359.47   857.1 2366.93
#Mann= 3 ,-1 , 0
       0      .1       0   374.7    .045       0   424.3      .1       0
#XS Ineff= 2 , 0
                          644.72          2360.5
Permanent Ineff=
       F       F
Bank Sta=374.7,424.3
XS Rating Curve= 0 ,0
Exp/Cntr=0.3,0.1

Type RM Length L Ch R = 1 ,50642   ,266,268.7,272
XS GIS Cut Line= 3
2395154.10886986670380.5797629962395638.02203531670423.056858749
2396037.06403531670462.358858749
#Sta/Elev= 30
       0 2423.45    68.9 2392.34   145.2 2361.72   169.3  2353.9   193.4 2341.86
   205.4 2341.79   217.5 2337.39   279.6 2341.31   301.7 2338.49   321.9 2340.85
   390.1 2342.43   410.2 2339.46   438.3 2339.34   454.4 2341.27   473.5 2339.59
   506.6 2338.08   511.9 2340.02   518.7 2343.52   562.9 2341.82   578.9 2346.63
     599 2348.56   687.5 2349.47   707.6 2359.77   727.5 2380.49   743.7 2393.08
   812.1 2436.72   832.2 2451.93   844.2 2456.73   856.3 2465.57   886.7 2481.63
#Mann= 4 ,-1 , 0
       0      .1       0   473.5    .045       0   511.9      .1       0
  801.34      .1       0
Bank Sta=473.5,511.9
XS Rating Curve= 0 ,0
Exp/Cntr=0.3,0.1

Type RM Length L Ch R = 1 ,50373   ,304.5,300,295
XS GIS Cut Line= 3
      2395194.05      670587.492      2395591.22      670687.233
     2395988.116      670788.047
#Sta/Elev= 30
       0 2396.33    23.2 2383.62      42 2371.46    54.3 2366.89    91.4 2338.43
    99.7  2334.5   145.1 2330.69   206.9  2334.7   297.7 2333.71     310 2331.05
   355.4  2335.1   389.1 2332.81   408.8 2329.85   421.4 2331.22   429.6 2334.66
   437.9 2335.76   491.6  2334.9   512.2 2332.93   516.3 2333.13   524.6 2337.11
   578.2    2340   627.7 2339.09   660.8 2340.36   693.8 2336.12   706.2 2336.67
   714.4 2339.07   722.7  2344.2   768.1 2381.78   780.4 2388.75     819 2405.87
#Mann= 3 ,-1 , 0
       0      .1       0   389.1    .045       0   429.6      .1       0
#XS Ineff= 2 , 0
                          594.46         2346.89
Permanent Ineff=
       F       F
Bank Sta=389.1,429.6
XS Rating Curve= 0 ,0
Exp/Cntr=0.3,0.1
