HEC-RAS study SENECACK.prj: SENECACK

--- SENECACK.g03 (geometry) --- (continued)

Type RM Length L Ch R = 1 ,20428   ,52.8,54.3,55.6
XS GIS Cut Line= 3
2416617.71665818678561.8868124672416413.06465818678207.193812467
2416208.41165818677852.499812467
#Sta/Elev= 30
       0 1900.28    24.9 1893.49      62 1874.03    74.7 1864.94    83.4 1856.81
     118 1832.05   132.8 1820.14   137.4 1813.74     142 1804.58   144.9 1800.45
   146.6 1798.57   150.8 1797.13   256.2 1799.87   271.3 1798.59   308.9 1798.98
   345.2  1798.2   358.1 1793.31   368.3 1790.92   423.1 1790.64   434.8 1793.45
   443.6 1797.59   451.4 1798.62   534.5 1799.87   569.6 1796.43   581.3  1798.5
   599.2 1809.77   682.3  1868.6   721.8 1900.22   786.3 1946.58     819  1973.7
#Mann= 6 ,-1 , 0
       0     .05       0    7.77      .1       0  216.94    .055       0
  321.52     .06       0   358.1    .045       0   434.8      .1       0
#XS Ineff= 2 , 0
             325    1797     454            1797
Permanent Ineff=
       F       F
Bank Sta=358.1,434.8
XS Rating Curve= 0 ,0
Exp/Cntr=0.5,0.3

Type RM Length L Ch R = 1 ,20373   ,152.2,145.5,140.2
XS GIS Cut Line= 2
2416645.98943728678531.4033414342416276.42620266677831.365291245
#Sta/Elev= 30
       0 1898.86    27.7  1890.8      82 1859.76    91.6  1847.1   109.4 1836.33
   130.1 1821.16     136 1815.22     144 1801.11   149.8 1797.08   201.1 1797.96
   217.7 1804.07   244.8 1804.79   262.9 1798.04   339.8 1797.43     348 1793.73
     361 1790.15   407.7 1789.67   416.7 1790.61   421.2 1793.23   426.1 1795.98
   434.8 1797.34   457.4 1795.77   512.5 1798.73   553.4 1795.22     566 1796.02
   584.1 1805.54   671.8 1861.34   710.3 1891.34   745.8 1921.81   791.6 1956.77
#Mann= 7 ,-1 , 0
       0      .1       0   83.55     .05       0  186.71     .06       0
   205.6    .055       0  289.87     .06       0     348    .045       0
   421.2      .1       0
#XS Ineff= 2 , 0
          239.84 1816.48
Permanent Ineff=
       F       F
Bank Sta=348,421.2
XS Rating Curve= 0 ,0
Exp/Cntr(USF)=0,0
Exp/Cntr=0.5,0.3

Type RM Length L Ch R = 1 ,20228   ,464.3,454.5,449.3
XS GIS Cut Line= 3
2416837.22202855678438.4189121332416589.06602855678112.674912133
2416340.91002855677786.930912133
#Sta/Elev= 30
       0 1898.35    74.8 1897.67    92.8 1896.35     107 1891.82   115.1  1887.9
   165.3 1852.38   198.4 1825.33   205.6  1818.4   221.2 1800.11   228.5 1796.08
   306.1 1797.06   321.2 1793.22   361.5 1793.02   369.6 1791.24   378.2 1788.85
   401.7 1787.66   433.1  1787.9   441.9 1791.09   446.9 1792.96   487.2 1790.31
   555.1 1790.27     578 1790.94   584.9 1792.73   617.9 1817.69   663.6 1841.98
   693.3 1855.55     717 1870.79   740.7 1888.88   778.8 1923.78     819 1956.01
#Mann= 6 ,-1 , 0
       0     .05       0   18.75      .1       0  240.66    .055       0
  351.62      .1       0   369.6    .045       0   441.9      .1       0
Bank Sta=369.6,441.9
XS Rating Curve= 0 ,0
Exp/Cntr=0.3,0.1

Type RM Length L Ch R = 1 ,19773   ,306.8,300,296.8
XS GIS Cut Line= 3
     2417232.347      678072.012     2416921.286      677805.682
     2416610.225      677539.353
#Sta/Elev= 30
       0  1855.3    21.8 1851.24    63.2 1839.66    81.4 1832.28      94 1822.47
   100.1 1819.73   124.7 1816.47   152.3 1797.47   160.1 1794.52   197.7 1792.47
   253.9 1785.11   316.8 1785.04   328.6  1786.2   344.4 1790.74   359.4 1782.99
   395.3 1778.96   419.9 1779.41   430.3 1783.06   450.7 1784.79   524.5 1782.42
   544.5 1783.61   586.3 1779.81   594.8 1780.57   604.5 1788.86   617.5 1806.55
   696.7 1867.97   734.1 1890.09   776.7 1910.86   804.8 1928.03     819 1939.77
#Mann= 5 ,-1 , 0
       0      .1       0  138.62     .06       0  267.07      .1       0
   359.4    .045       0   430.3      .1       0
#XS Ineff= 2 , 0
          343.94 1802.61
Permanent Ineff=
       F       F
Bank Sta=359.4,430.3
XS Rating Curve= 0 ,0
Exp/Cntr=0.3,0.1

Type RM Length L Ch R = 1 ,19473   ,301.9,300,296.4
XS GIS Cut Line= 3
     2417442.549      677780.526     2417095.821      677562.651
     2416749.092      677344.775
#Sta/Elev= 30
       0 1831.75    37.6 1827.89    61.2 1823.38    73.6 1818.56    93.9 1806.97
   140.3 1783.95   217.1 1780.38     326 1780.04   339.9 1780.62   358.8 1784.88
     373 1780.44   382.4 1777.06   391.9 1776.73   444.9 1776.88     458 1779.92
   505.3 1778.01   519.4 1775.25   533.6 1774.82   544.4 1776.25   557.2 1783.11
   576.1 1799.36     597    1813   639.3 1844.84   642.3 1847.48   650.9 1859.97
   662.5 1867.54   694.7 1881.83   761.1 1908.39   769.9 1910.64     819 1935.34
#Mann= 5 ,-1 , 0
       0      .1       0   67.98     .06       0  216.72      .1       0
     373    .045       0     458      .1       0
Bank Sta=373,458
XS Rating Curve= 0 ,0
Exp/Cntr=0.3,0.1

Type RM Length L Ch R = 1 ,19173   ,294.3,300,311.9
XS GIS Cut Line= 3
     2417598.401      677504.237     2417242.541      677301.171
     2416881.001      677108.953
#Sta/Elev= 30
       0    1793      18 1787.61      35 1780.69    51.1 1777.96    83.4 1777.96
   100.4 1780.01   115.1 1780.25   156.1 1777.62   228.7  1778.2   312.8 1773.92
   372.6 1777.45   377.2 1777.18   384.9 1773.42   390.7 1771.67   423.1 1770.94
   450.3 1771.49   458.6 1773.13     482 1772.64   508.9 1776.81   522.7 1780.94
     559 1796.05   622.4 1815.37   685.8 1833.67   708.5 1841.37   749.3 1850.79
   783.9 1862.06   795.8 1864.07   803.6 1867.36   812.7 1873.03   819.2 1875.01
#Mann= 4 ,-1 , 0
       0     .06       0  141.41      .1       0   384.9    .045       0
   458.6      .1       0
Bank Sta=384.9,458.6
XS Rating Curve= 0 ,0
Exp/Cntr=0.3,0.1

Type RM Length L Ch R = 1 ,18873   ,560.8,552.2,542.9
XS GIS Cut Line= 3
      2417735.23      677348.783     2417433.601      677071.817
     2417131.973      676794.851
#Sta/Elev= 30
       0 1814.86    11.5 1800.58    16.9 1796.71      47 1780.21      64  1774.9
   100.8 1774.76   120.1 1776.86   141.9 1776.92     163 1774.72   201.6 1775.38
     265 1773.12   310.3 1774.19   330.1 1773.16   345.8 1769.49   366.9 1767.72
   393.1 1763.74   434.5 1763.84     449 1768.08   499.6 1778.43   511.3 1783.63
   538.3 1799.88   564.6 1806.67   613.2 1813.71   629.7 1817.59   652.8 1820.57
   736.1 1835.56   753.9 1841.18   783.5 1848.23   797.2 1853.31     819 1857.49
#Mann= 5 ,-1 , 0
       0      .1       0   63.03     .06       0  192.71      .1       0
   366.9    .045       0     449      .1       0
Bank Sta=366.9,449
XS Rating Curve= 0 ,0
Exp/Cntr=0.3,0.1

Type RM Length L Ch R = 1 ,18321   ,131.3,126.4,123.4
XS GIS Cut Line= 3
2417984.60790187676987.5621859942417956.26289407676744.222273532
2417352.48319224676422.685644067
#Sta/Elev= 30
       0 1838.16    28.9 1835.46      53 1828.71    93.3 1803.11   113.4 1788.33
   129.5 1783.55   145.6 1774.48   181.9 1774.31     202 1777.35   226.2 1775.24
   251.2 1772.91   273.9 1766.15   319.2 1763.74   364.5 1764.73   381.2 1759.06
   403.8 1756.31   446.1 1756.56   452.1 1758.73   459.7 1764.95   468.8 1765.69
   483.7 1762.92   542.8  1760.9   695.4 1760.66   844.9 1760.03   862.2 1766.69
   876.6 1780.24   890.2 1796.35   903.8 1805.82   917.4 1811.17     929 1818.93
#Mann= 7 ,-1 , 0
       0      .1       0    28.9     .06       0   226.2    .055       0
   319.2     .05       0   381.2    .045       0   452.1     .05       0
   695.4      .1       0
#XS Ineff= 2 , 0
                           468.4            1778
Permanent Ineff=
       F       F
Bank Sta=381.2,452.1
XS Rating Curve= 0 ,0
Exp/Cntr=0.5,0.3

Type RM Length L Ch R = 1 ,18195   ,37.3,36.8,36.1
XS GIS Cut Line= 3
2418098.65235426 676709.640882442417977.82717018676597.605206344
 2417388.0156345676389.179003217
#Sta/Elev= 30
       0 1771.57    89.6 1770.69   114.4 1771.09     168 1766.14   184.9 1764.69
   223.2 1763.56   227.4 1762.59   233.31758.877   240.2 1755.31   248.6 1753.91
   286.8 1754.39   291.1 1755.27   296.6 1758.82   299.6 1761.03   304.1 1762.24
   329.2 1760.81   439.6 1758.99   562.6 1759.08   620.7 1760.03   655.9 1760.16
   716.5 1757.74   740.8 1757.42   749.3 1757.94   757.7 1759.84     762 1761.78
   766.2 1765.53   770.5  1771.4   774.7 1774.68   783.2 1779.12   790.3 1785.32
#Mann= 5 ,-1 , 0
       0      .1       0     168     .06       0   233.3    .045       0
   296.6     .05       0   620.7      .1       0
#XS Ineff= 2 , 0
             218    1768   304.1            1768
Permanent Ineff=
       F       F
Bank Sta=233.3,296.6
XS Rating Curve= 0 ,0
Exp/Cntr(USF)=0,0
Exp/Cntr=0.5,0.3

Type RM Length L Ch R = 1 ,18158   ,189.5,183.9,179.8
XS GIS Cut Line= 3
2418142.53965343676685.5737305962418002.67679286676565.254240378
2417362.76936592676352.611129318
#Sta/Elev= 30
       0  1770.1   139.1 1768.26   222.4 1764.69   256.1 1762.93   264.5    1761
   268.6  1759.2   277.2 1754.08   306.5 1753.42   323.5 1754.06   328.7  1757.6
   331.8 1760.16   336.2 1761.74   340.4 1761.97   360.3 1760.44   433.1 1758.75
   626.1 1758.34   669.2 1759.43   686.7 1761.23   702.9  1759.2   715.5 1758.49
     783 1756.58   795.6 1758.97   803.2 1761.63   808.3 1764.64   812.5 1769.45
   816.7 1776.41   820.9 1782.25   825.1 1786.58   841.2  1799.4   858.8 1810.67
#Mann= 6 ,-1 , 0
       0      .1       0   222.4     .06       0   268.6    .045       0
   328.7     .06       0   331.8     .05       0   669.2      .1       0
#XS Ineff= 2 , 0
                           340.4            1768
Permanent Ineff=
       F       F
Bank Sta=268.6,328.7
XS Rating Curve= 0 ,0
Exp/Cntr=0.5,0.3

Type RM Length L Ch R = 1 ,17974   ,321.8,300.6,280.4
XS GIS Cut Line= 3
2418254.11848846676480.5807475352417977.86327023676352.888921885
2417389.88377003676330.183943648
#Sta/Elev= 30
       0 1814.16      61 1804.92    78.6 1803.43    96.3 1803.41   105.1  1801.9
   137.5 1787.95   144.7 1782.95   157.9 1771.73     180 1763.73   184.4 1762.96
   281.3    1762   347.5 1763.42   355.5  1762.5   359.5 1761.28   363.8 1758.56
   371.5 1753.79   375.5 1753.29   431.6 1752.89   447.6 1753.64   459.6 1758.37
   459.6 1758.38   463.6 1758.83   476.2 1756.82   503.6 1756.16   727.8 1758.15
   839.9  1755.6   847.9 1757.84   875.9 1774.39   887.9 1784.72   892.8 1790.05
#Mann= 7 ,-1 , 0
       0      .1       0   99.51      .1       0  233.54     .06       0
  345.79      .1       0   363.8    .045       0   459.6     .05       0
  751.08      .1       0
Bank Sta=363.8,459.6
XS Rating Curve= 0 ,0
Exp/Cntr=0.3,0.1

Type RM Length L Ch R = 1 ,17673   ,257.6,263,263.8
XS GIS Cut Line= 3
     2418149.384      675905.313     2417772.061      676064.429
2417343.15729573676249.964385115
#Sta/Elev= 30
       0 1852.57      81 1843.22     104 1838.06   119.3 1832.61   128.8 1827.46
   143.7 1816.91   163.5 1793.41   176.5 1781.44   198.6 1764.44   211.2 1757.06
   232.9 1755.88     275 1757.25   293.7 1753.27   329.9 1754.13   363.2 1752.36
   371.9 1750.18   393.6 1749.97   441.4 1750.09     456 1752.35   464.1 1754.42
     485 1753.39   546.7 1754.05   694.2 1752.65   759.6 1756.78   768.3 1758.87
   794.5 1770.78     817 1784.78   855.5 1814.81   868.1 1830.17   876.8 1835.98
#Mann= 7 ,-1 , 0
       0      .1       0  187.56     .06       0  289.77      .1       0
   363.2    .045       0     456      .1       0  494.37     .05       0
  596.81      .1       0
Bank Sta=363.2,456
XS Rating Curve= 0 ,0
Exp/Cntr=0.3,0.1

Type RM Length L Ch R = 1 ,17410   ,306.4,337,357.9
XS GIS Cut Line= 3
      2418052.95      675695.2832417659.20292341675827.166714904
     2417277.279      675976.119
#Sta/Elev= 30
       0 1820.85     2.3  1819.1     6.5 1812.28    14.1 1796.14    23.4 1784.27
    52.9 1770.13    61.4 1762.02    69.8 1756.83    78.3 1752.95    86.7 1751.59
   127.8 1752.48   171.1 1752.26   196.4 1754.12   225.5 1752.79   323.8 1753.24
   335.6  1752.5   348.2 1747.84   356.7 1745.61     420 1744.75   445.8 1747.48
   510.2 1746.77   557.4 1754.26     566 1757.09   600.7 1783.92   621.8 1797.41
   707.7 1842.53   779.9 1884.81   797.9 1899.95     815 1919.23   825.2 1926.71
#Mann= 5 ,-1 , 0
       0      .1       0   127.8    .055       0   225.5      .1       0
   348.2    .045       0   445.8      .1       0
#XS Ineff= 2 , 0
           196.4    1760
Permanent Ineff=
       F       F
Bank Sta=348.2,445.8
XS Rating Curve= 0 ,0
Exp/Cntr=0.3,0.1

Type RM Length L Ch R = 1 ,17073   ,285.7,300,312.9
XS GIS Cut Line= 3
2418085.06458299675651.302110651     2417653.394      675511.182
     2417272.814      675362.049
#Sta/Elev= 30
       0  1811.8    19.3 1798.65    31.9 1785.71    43.4 1776.59    78.1 1754.61
    86.5 1751.42   183.3 1749.22   212.7 1751.98   229.5 1747.11   250.6 1745.62
   372.5 1746.55   392.7 1744.76   406.2 1739.91   418.8 1739.73   428.9 1742.03
   440.3 1740.35   486.3  1740.8   499.6 1755.44   539.5 1779.59   568.4 1802.09
   592.2 1817.89   645.7 1849.24     693 1872.69   710.2 1883.96   755.5 1908.61
   761.7 1913.17   778.9 1931.68     809 1951.28   830.5  1962.8   862.6  1985.1
#Mann= 5 ,-1 , 0
       0      .1       0  179.23    .055       0  290.89      .1       0
   428.9    .045       0   486.3      .1       0
Bank Sta=428.9,486.3
XS Rating Curve= 0 ,0
Exp/Cntr=0.3,0.1

Type RM Length L Ch R = 1 ,16773   ,450,450,449.2
XS GIS Cut Line= 3
     2418100.893      675519.533     2417791.968      675250.245
     2417493.147      674970.333
#Sta/Elev= 30
       0  1791.8     2.8 1786.65     4.8 1785.18    37.5 1766.56    55.8 1752.14
    61.2 1750.13    92.7 1748.22   251.5 1746.44   289.4    1741   342.5 1739.97
   360.1  1742.3     369 1739.05   407.4 1736.48     447 1739.19   469.7 1754.07
   493.7 1775.44   504.7 1783.16   520.6  1804.6   555.1 1838.95   602.7 1873.02
   607.8 1881.02   619.5 1909.11   625.2 1916.73   641.7  1932.2   681.9 1963.23
   715.9 1993.39   738.5  2017.1   748.2 2029.59   789.4 2070.56   819.3 2090.91
#Mann= 6 ,-1 , 0
       0      .1       0   74.94     .06       0  151.53    .055       0
  202.43      .1       0     369    .045       0     447      .1       0
Bank Sta=369,447
XS Rating Curve= 0 ,0
Exp/Cntr=0.3,0.1

Type RM Length L Ch R = 1 ,16323   ,483,484.8,489.6
XS GIS Cut Line= 3
     2418404.288      675185.958      2418094.95      674917.629
     2417785.612        674649.3
#Sta/Elev= 30
       0 1813.63    29.1  1793.1    49.7 1789.63    65.7 1777.12    96.2 1759.88
   139.7 1741.31   182.1 1741.81   201.8 1738.45   261.3 1735.22   360.5 1737.79
   374.7 1736.33   383.3 1732.27   403.1 1730.91   462.7 1733.16   480.8 1736.88
   526.3 1761.65   593.1 1805.33   600.4 1816.15     611 1839.13   615.7 1845.88
   646.9 1868.15   663.9 1905.55   678.1 1922.94   695.1 1939.21   726.3 1962.57
   743.3 1979.52   763.2 1995.36   780.4 2014.56   805.7 2037.09     819 2046.51
#Mann= 5 ,-1 , 0
       0      .1       0   87.64     .06       0   236.8      .1       0
   374.7    .045       0   480.8      .1       0
Bank Sta=374.7,480.8
XS Rating Curve= 0 ,0
Exp/Cntr=0.3,0.1

Type RM Length L Ch R = 1 ,15839   ,235.4,429.9,488.2
XS GIS Cut Line= 3
2418578.42823629674980.6549030072418484.36796221674621.482197086
2418163.45236328674314.237494125
#Sta/Elev= 30
       0 1849.75    47.1 1842.15    60.2 1838.04   101.1 1817.03   109.3  1811.4
   117.6 1808.34   134.1 1797.13     188 1775.16     192 1772.42   196.2 1767.44
   204.4 1748.87   207.6 1743.15   214.2 1738.25   286.3 1736.63   328.9  1730.4
   403.91731.552   409.7 1730.49   421.3 1724.36   434.4 1723.11   481.21725.078
   495.4 1733.27   512.9 1748.87   518.5 1752.37   561.8 1763.76   589.5 1767.37
   606.1 1777.67   631.7 1790.32     660  1806.7   716.9 1836.63   815.6 1864.35
#Mann= 6 ,-1 , 0
       0      .1       0  208.73     .06       0  336.05      .1       0
   403.9    .045       0   481.2    .045       0   516.3      .1       0
Bank Sta=403.9,481.2
XS Rating Curve= 0 ,0
Exp/Cntr=0.5,0.3

Type RM Length L Ch R = 1 ,15409   ,236.8,152,180.5
XS GIS Cut Line= 4
2418639.20144195675016.4189085972418532.31480156674558.462059695
2418947.03393344674173.352836458  2418999.495913673914.062273389
#Sta/Elev= 30
       0 1855.31    50.9 1853.75      96 1848.26   141.5  1836.6   211.5 1799.78
   268.1 1779.67   278.1  1770.5   293.2 1747.76     308  1736.7   391.8 1736.43
   424.6  1733.9   461.6 1726.28   545.3 1726.29   624.91721.927     840 1717.43
     851 1718.36   857.51722.338   866.6 1725.53   928.1 1728.59   998.7 1736.62
  1017.9 1735.17  1042.8 1726.28  1067.3 1725.05  1128.5 1740.66  1136.7 1748.49
  1144.8 1764.75  1157.4 1780.28    1218 1828.74  1268.9 1886.12  1300.8 1907.02
#Mann= 13 ,-1 , 0
       0      .1       0   91.25     .06       0  311.57      .1       0
  326.17     .06       0   435.2      .1       0  486.45     .06       0
  569.34      .1       0   624.9    .045       0   857.5    .045       0
     860    .055       0  939.15      .1       0 1174.84     .06       0
 1245.23      .1       0
#XS Ineff= 2 , 0
             525    1736     874            1735
Permanent Ineff=
       F       F
Bank Sta=624.9,857.5
XS Rating Curve= 0 ,0
Exp/Cntr=0.5,0.3

Type RM Length L Ch R = 1 ,15257   ,482.1,433.3,369.6
XS GIS Cut Line= 5
2418710.95193715 674964.700095232418677.60065109674700.921741837
 2418844.9859094674421.8762063862419114.67495999674256.743914196
2419176.70953336673955.083216749
#Sta/Elev= 30
       0 1860.33    42.1 1856.08   134.9 1840.26   163.4 1828.71   231.6 1797.12
   394.2 1768.13   426.8  1756.3   454.7 1759.15   507.3 1758.81   571.4 1740.71
   571.4 1740.67   571.4 1740.65   579.1 1730.93   591.3 1723.26   625.31719.321
   711.1 1714.64   764.41718.708   819.1 1722.15   850.7 1719.33   888.1 1720.57
   954.3 1730.21  1003.3 1733.25  1052.3 1719.99  1068.3 1724.68  1089.1 1732.46
  1125.7 1736.48  1150.3 1751.01  1162.6 1766.85  1178.9 1800.67  1215.5 1835.49
#Mann= 11 ,-1 , 0
       0      .1       0    42.1     .06       0   134.9      .1       0
   163.4     .06       0   454.7    .055       0   571.4    .045       0
   625.3    .045       0   764.4    .055       0   850.7     .06       0
   954.3    .035       0  1068.3    .055       0
#XS Ineff= 2 , 0
                           999.2            1740
Permanent Ineff=
       F       F
Bank Sta=625.3,764.4
XS Rating Curve= 0 ,0
Exp/Cntr=0.5,0.3

Type RM Length L Ch R = 1 ,14823   ,585.7,600,622
XS GIS Cut Line= 3
     2419308.561      674820.056     2419354.523      674413.143
     2419400.485      674006.231
#Sta/Elev= 30
       0  1877.6    73.6 1859.07   210.5  1830.3   226.6 1825.05   245.4 1810.75
   266.9  1809.1     283 1794.85     287 1786.72     291 1773.64     295 1765.36
   319.2 1744.93   339.3 1721.73   363.5 1718.72     372 1712.43   379.6 1710.53
   407.3 1710.38   469.6 1712.63   488.3 1713.57   512.4  1719.1     609 1723.89
   669.4    1729   681.5 1727.36   705.6 1719.62   717.7  1719.4   733.8 1725.05
   741.9  1729.6   780.7 1758.84   787.9 1765.79   798.7 1782.88     819    1804
#Mann= 8 ,-1 , 0
       0      .1       0  141.83     .06       0  329.38      .1       0
     372    .045       0   469.6    .035       0  647.38    .055       0
  697.46    .035       0   748.5      .1       0
#XS Ineff= 2 , 0
                          679.67          1739.2
Permanent Ineff=
       F       F
Bank Sta=372,469.6
XS Rating Curve= 0 ,0
Exp/Cntr=0.3,0.1

Type RM Length L Ch R = 1 ,14223   ,299,300,299.4
XS GIS Cut Line= 4
     2419701.065      675025.066     2419883.817       674658.75
  2419912.045454674609.682606537   2419800.82683674128.390147888
#Sta/Elev= 30
       0 1852.65    11.8 1847.54    24.8 1840.84    42.7 1837.96    84.4 1812.02
    96.3 1801.99   114.2 1780.22   123.1    1766   132.1 1759.02   178.8 1728.06
     217 1709.45   344.2 1707.96     369 1712.04   382.4 1704.58   400.3 1701.15
   436.81704.016   493.5 1705.46     514  1704.9   530.4 1709.36   555.1 1710.38
     707  1717.4   789.1  1716.3   820.4 1720.21   838.3  1729.3   854.8 1742.39
   867.1 1768.17   909.6 1797.84   924.5 1824.14   928.7 1829.03     960 1842.95
#Mann= 7 ,-1 , 0
       0      .1       0    11.8     .06       0   132.1      .1       0
   382.4    .045       0   436.8      .1       0   493.5    .055       0
   555.1     .06       0
#XS Ineff= 2 , 0
           364.5    1720
Permanent Ineff=
       F       F
Bank Sta=382.4,436.8
XS Rating Curve= 0 ,0
Exp/Cntr=0.3,0.1

Type RM Length L Ch R = 1 ,13923   ,444.6,450,451.9
XS GIS Cut Line= 3
     2419954.583      675156.239     2420150.262      674796.517
     2420345.942      674436.795
#Sta/Elev= 30
       0 1840.37     6.1 1835.69    24.3 1819.55    28.9 1800.53    33.4 1774.67
      38  1761.8     122 1707.92   151.8 1704.58   195.8 1706.17   224.7 1703.14
   302.1 1702.75   352.2 1704.04   365.8 1708.86   375.7 1704.32   381.6 1700.11
   388.6  1698.8   440.5 1701.67   470.5 1700.83   484.2 1705.71   490.7 1705.53
   593.5 1709.43   614.6 1717.75     652 1717.57   658.8  1716.9     680 1724.54
   707.3 1747.94   716.4 1752.51     721  1752.4   730.1 1760.05     819 1807.26
#Mann= 9 ,-1 , 0
       0     .06       0     6.1      .1       0   375.7    .045       0
   440.5      .1       0   470.5    .035       0   490.7      .1       0
   593.5     .06       0     652    .055       0   716.4      .1       0
#XS Ineff= 2 , 0
           365.8    1720
Permanent Ineff=
       F       F
Bank Sta=375.7,440.5
XS Rating Curve= 0 ,0
Exp/Cntr=0.3,0.1

Type RM Length L Ch R = 1 ,13473   ,393.1,382.1,387.6
XS GIS Cut Line= 3
     2420297.565      675360.804     2420536.623      675026.939
     2420751.999      674678.887
#Sta/Elev= 30
       0 1833.82      28 1811.51    31.9 1805.78    36.8 1792.73    41.7 1783.96
    91.1 1741.29   125.3 1706.15   135.2 1699.88   154.2 1697.47   282.8 1697.06
   302.5 1698.08   317.2 1701.76   346.7 1696.65     450 1696.79   473.2 1695.59
   495.4 1701.74   508.1 1698.01   556.5 1703.49   575.3 1703.27   617.7 1725.27
   674.1 1719.45   697.6 1725.09   716.4 1733.92   744.7  1734.9   758.8 1737.66
   763.5 1739.38   801.1  1771.7   810.5 1787.21   815.2 1789.26   819.9  1788.2
#Mann= 4 ,-1 , 0
       0      .1       0   346.7    .045       0     450      .1       0
  594.52     .06       0
Bank Sta=346.7,450
XS Rating Curve= 0 ,0
Exp/Cntr=0.3,0.1

Type RM Length L Ch R = 1 ,13091   ,393.3,367.9,360.6
XS GIS Cut Line= 2
2420657.24578717675600.0123128512420995.60222977674938.444131916
#Sta/Elev= 30
       0 1918.35    28.2 1907.94    40.6 1898.91    61.4 1897.87     145 1845.92
   149.5 1840.42   158.5 1816.21     163 1809.35     181 1795.12   201.4 1774.98
   252.9 1734.83   261.8 1725.22   270.8 1709.33   284.3 1693.89   284.3 1693.87
   297.8 1688.67   324.7 1688.36   355.7  1689.2   367.6 1691.63   441.9 1694.87
   498.4  1692.2   576.3 1692.76   612.3 1698.06   639.2 1707.43   652.7  1725.4
   661.8 1731.33   693.2  1737.9   714.8 1738.79   724.3 1742.24   743.1 1739.74
#Mann= 4 ,-1 , 0
       0     .06       0  125.34      .1       0   284.3    .045       0
   367.6      .1       0
Bank Sta=284.3,367.6
XS Rating Curve= 0 ,0
Exp/Cntr=0.3,0.1

Type RM Length L Ch R = 1 ,12723   ,472.4,450,423.9
XS GIS Cut Line= 3
      2421154.82      675768.956     2421167.798      675359.662
     2421180.776      674950.368
#Sta/Elev= 30
       0 1899.02    21.3 1895.69    46.1 1887.98    82.1 1880.17   102.1 1873.27
   126.1  1862.5   138.1  1854.8   150.1 1843.56   178.2 1823.88   190.2 1806.25
   254.2 1757.83   294.2 1715.32   322.2 1687.76   330.2 1685.58   374.2 1685.69
   410.3 1684.45   426.3 1684.94   434.3 1687.45   446.3  1689.3   534.3 1688.55
   566.3 1689.84   586.4 1689.75   614.4  1686.7   638.4 1690.03   706.4 1691.32
   722.4 1699.69   730.4 1702.34   766.5 1704.78   774.5 1710.61     819 1731.66
#Mann= 6 ,-1 , 0
       0      .1       0   38.36      .1       0  190.78      .1       0
   374.2    .045       0   434.3      .1       0  786.27     .06       0
Bank Sta=374.2,434.3
XS Rating Curve= 0 ,0
Exp/Cntr=0.3,0.1

Type RM Length L Ch R = 1 ,12273   ,452.3,450,447.3
XS GIS Cut Line= 3
     2421797.117      675695.444     2421609.408      675332.212
2421399.38380192674915.864385071
#Sta/Elev= 30
       0 1934.41    18.6 1923.49    32.1  1908.7    72.7 1882.58    85.3 1870.22
   106.1 1856.43   180.3 1802.21   216.7 1773.17   275.3 1730.97   319.8 1695.76
   333.8 1687.43   360.8 1683.18   369.8 1680.27   379.8 1679.77   428.3 1679.98
   464.1 1682.11   516.1 1684.53   562.7  1682.5   593.5 1678.75   620.9  1685.4
   665.7 1686.09   679.2 1683.46   741.9 1686.27   782.2 1685.04   795.6 1686.91
   800.1 1688.65     818 1701.36   828.7 1707.46   858.8 1722.82   875.2  1729.6
#Mann= 4 ,-1 , 0
       0      .1       0   360.8    .045       0   464.1      .1       0
  840.82     .06       0
Bank Sta=360.8,464.1
XS Rating Curve= 0 ,0
Exp/Cntr=0.3,0.1

Type RM Length L Ch R = 1 ,11823   ,299.4,300,295.4
XS GIS Cut Line= 3
     2422209.317      675469.563     2422003.618      675115.475
     2421797.919      674761.387
#Sta/Elev= 30
       0 1796.17    33.1    1772    58.6 1744.52   103.3 1714.68   129.7 1709.38
   148.5 1701.96   191.1 1691.83   217.4 1681.35   240.9 1678.23   299.8 1678.98
   317.7 1676.52   331.6 1678.65   377.8 1675.39   395.9 1673.37   430.8 1673.23
   451.1 1676.22     472 1678.39   502.7 1673.66   527.6 1673.11   541.2 1673.95
   562.8  1680.2   597.8 1679.25   618.3 1682.14   627.6 1685.76   713.8 1732.08
   738.6 1741.97   757.1 1747.02   777.5 1757.67   784.9 1759.25     819 1758.12
#Mann= 5 ,-1 , 0
       0      .1       0   377.8    .045       0   451.1      .1       0
  685.73     .06       0  802.77      .1       0
Bank Sta=377.8,451.1
XS Rating Curve= 0 ,0
Exp/Cntr=0.3,0.1

Type RM Length L Ch R = 1 ,11523   ,300.9,300,299.4
XS GIS Cut Line= 3
2422520.98938507675364.150424241     2422275.299      674991.553
     2422042.948      674646.464
#Sta/Elev= 30
       0 1811.97    34.3 1793.42    68.6 1771.78    89.2 1756.56   106.5 1740.24
   111.7 1731.65     118 1718.27   126.1 1707.14   149.4 1689.06   169.2 1678.53
   212.3 1673.56   413.6 1675.88   425.5  1672.9   432.8 1668.68   440.1 1668.28
   468.8 1669.25   493.3 1672.78   513.5  1673.7     558 1667.25   572.5 1669.21
   582.6 1679.93   614.3 1708.05   647.8 1724.66   717.2 1745.05   731.6 1746.19
   790.1 1760.97   804.5 1757.47   837.7 1756.86   848.4 1762.54   862.3 1774.09
#Mann= 5 ,-1 , 0
       0      .1       0   425.5    .045       0   493.3      .1       0
  749.07     .06       0   856.8      .1       0
#XS Ineff= 2 , 0
           411.7 1682.73
Permanent Ineff=
       F       F
Bank Sta=425.5,493.3
XS Rating Curve= 0 ,0
Exp/Cntr=0.3,0.1

Type RM Length L Ch R = 1 ,11223   ,280.3,300,323.8
XS GIS Cut Line= 3
2422782.31329859675147.848418029     2422482.422       674775.05
2422251.36790835674484.775837399
#Sta/Elev= 30
       0 1708.51    48.7  1677.6    57.7 1674.39    78.2 1671.54   134.7 1668.03
   333.2 1671.04   356.7 1669.43   373.1 1670.39   390.1 1667.81   411.9 1670.05
   449.9 1668.15   463.3 1663.29     494  1662.7   543.8 1665.95   560.9 1664.86
   566.6 1665.97   580.7 1672.78   612.8 1692.19   642.3 1706.13   664.2 1722.21
     689 1746.68   702.7 1755.39   739.4 1757.05   768.7 1760.53   786.2 1757.53
   805.5 1759.61   816.1 1768.39   825.6 1771.39   836.5 1777.56   849.5 1779.72
#Mann= 5 ,-1 , 0
       0      .1       0   449.9    .045       0   543.8      .1       0
  696.62     .06       0  808.89      .1       0
Bank Sta=449.9,543.8
XS Rating Curve= 0 ,0
Exp/Cntr=0.3,0.1

Type RM Length L Ch R = 1 ,10923   ,447.2,450,451
XS GIS Cut Line= 3
2422860.30956721675151.204612171     2422752.153      674651.903
     2422670.284       674250.68
#Sta/Elev= 30
       0 1741.77    61.1 1691.18      74 1674.82    94.5 1668.76   131.3 1670.87
   233.6 1665.66   311.4 1668.31   352.3 1665.37   438.2    1667   447.7 1664.68
     471 1659.44   536.4 1660.03   543.4 1665.18   557.9 1676.38   607.9 1703.94
   642.6 1726.01   687.5  1762.7     696 1765.75   728.3 1767.14   741.2 1780.15
   760.4 1804.61   773.2  1813.8   785.4 1828.97   818.1 1849.99   830.3 1867.78
   871.2 1901.09   875.3 1905.84   883.4 1919.95   891.6 1929.19   920.4 1951.29
#Mann= 5 ,-1 , 0
       0      .1       0   447.7    .045       0   543.4      .1       0
  620.26     .06       0  717.91      .1       0
Bank Sta=447.7,543.4
XS Rating Curve= 0 ,0
Exp/Cntr=0.3,0.1

Type RM Length L Ch R = 1 ,10473   ,442.5,450,459.5
XS GIS Cut Line= 3
      2423263.59      674996.386     2423197.914      674592.187
     2423132.239      674187.988
#Sta/Elev= 30
       0 1702.89     9.6 1696.03    33.9 1674.38    46.1 1666.46    54.2 1664.34
   106.9  1662.1   179.9    1664   232.5 1661.19   285.2 1660.77   301.4 1657.67
   322.8 1662.02   374.3 1662.93     382 1661.84   385.5 1659.21   390.6 1655.21
   394.6  1654.6   434.3 1654.44   455.4 1655.24   463.5 1660.08   479.8 1676.37
   564.8  1739.5   621.5 1788.79   629.6  1792.8     658 1793.57   667.9 1805.23
   682.3 1817.93   690.4 1830.12   706.6 1851.35   783.6  1911.4     819 1940.78
#Mann= 5 ,-1 , 0
       0      .1       0   385.5    .045       0   463.5      .1       0
  625.74     .06       0  723.28      .1       0
Bank Sta=385.5,463.5
XS Rating Curve= 0 ,0
Exp/Cntr=0.3,0.1

Type RM Length L Ch R = 1 ,10023   ,445.1,450,456.1
XS GIS Cut Line= 3
     2423636.988      674950.298     2423643.602      674540.852
     2423650.216      674131.405
#Sta/Elev= 30
       0 1692.95    83.4  1681.3   155.4 1678.81   187.4 1664.74   211.4 1656.17
   327.4 1655.71   356.4 1653.37   391.5 1651.25   455.5  1651.5   465.2  1654.6
   471.5 1660.48   487.5 1683.81   519.5 1711.37   546.5 1742.19   575.5 1771.36
   579.5  1776.7   591.5 1805.11   595.6 1812.59   607.5 1818.97   631.5 1837.15
   643.5 1842.51   651.5 1842.67   667.5  1837.5   695.5  1836.2   703.5 1838.51
   711.5 1848.21   731.5 1884.97   739.5 1895.55   743.5 1898.31     819 1925.77
#Mann= 5 ,-1 , 0
       0      .1       0   356.4    .045       0   465.2      .1       0
  646.87     .06       0  745.84      .1       0
Bank Sta=356.4,465.2
XS Rating Curve= 0 ,0
Exp/Cntr=0.3,0.1

Type RM Length L Ch R = 1 ,9573    ,458.5,444.2,446.3
XS GIS Cut Line= 3
     2424048.942      675006.991     2424087.928       674599.35
     2424126.915      674191.711
#Sta/Elev= 30
       0  1686.8     8.1 1684.44   136.7 1670.74   156.8 1665.45   180.9 1655.31
   188.8 1653.67   346.5 1652.81   353.7  1652.6   361.7  1648.8   365.8 1646.58
   372.2 1645.08   408.8 1644.55   442.1 1646.88   482.3 1650.64   522.5  1649.5
   542.6 1646.66   550.6  1647.2     558 1651.48   570.7 1663.93   580.2 1668.88
   586.8 1674.24   590.8 1679.28   610.9 1710.91     639 1741.27   671.1 1765.91
   687.2 1775.75   694.9 1778.48   715.3 1781.93   768.3 1783.51     819 1789.71
#Mann= 3 ,-1 , 0
       0      .1       0   361.7    .045       0   442.1      .1       0
Bank Sta=361.7,442.1
XS Rating Curve= 0 ,0
Exp/Cntr=0.3,0.1

Type RM Length L Ch R = 1 ,9129    ,345.3,305.8,293.3
XS GIS Cut Line= 3
     2424372.664       675142.692424470.88061124674952.565626011
     2424534.649      674296.417
#Sta/Elev= 30
       0 1803.48    35.8 1788.95   123.1 1750.56   155.8 1739.19     214  1712.1
   229.4 1703.02   255.9 1685.45     276 1670.71   292.3 1657.62   312.1 1644.39
   316.1 1642.56   328.2 1640.42   396.5 1639.74   420.5 1640.29   429.7 1643.27
   436.7 1647.05   448.8 1647.75     501  1646.6   573.4    1648   629.6 1647.43
   637.7 1649.91   641.7 1653.15   654.9 1661.02   681.9 1674.28   693.9  1674.9
     706 1678.91   726.1 1682.35   778.3 1689.25   802.4 1691.35   873.2  1702.7
#Mann= 6 ,-1 , 0
       0      .1       0   312.1    .045       0   429.7      .1       0
  503.16      .1       0  525.73      .1       0  704.55      .1       0
Bank Sta=312.1,429.7
XS Rating Curve= 0 ,0
Exp/Cntr=0.3,0.1

Type RM Length L Ch R = 1 ,8823    ,488.9,450,418.5
XS GIS Cut Line= 3
2424932.88968084675061.492531928     2424758.091       674662.14
     2424612.531        674276.1
#Sta/Elev= 30
       0 1957.48      29 1937.39    52.2 1924.48    59.6 1917.68    72.7 1912.06
    94.5 1888.83   107.6 1877.73   120.7 1858.53   128.1  1851.2   190.6 1803.93
     195 1798.09   203.7 1780.92   208.1 1775.68   261.8 1722.41   267.8 1712.35
   277.9 1687.99   282.3 1682.73   316.4 1656.77   334.7 1651.11   364.5 1637.72
   408.9 1638.99   437.9 1635.22   465.1 1636.37   472.1 1640.21   478.3 1643.57
   606.1 1644.51   667.7 1647.46   708.7 1658.86   755.7  1663.5   848.5    1679
#Mann= 5 ,-1 , 0
       0      .1       0   364.5    .045       0   472.1      .1       0
  573.62      .1       0  697.54      .1       0
Bank Sta=364.5,472.1
XS Rating Curve= 0 ,0
Exp/Cntr=0.3,0.1

Type RM Length L Ch R = 1 ,8373    ,447.1,450,451.3
XS GIS Cut Line= 3
      2425471.43      674563.821     2425097.177      674399.476
2424724.56298581674225.610364079
#Sta/Elev= 30
       0 1934.62    42.1 1907.06    53.2  1893.4    70.6 1883.47    79.4 1883.25
    83.8 1880.41    95.3 1858.13   101.2 1851.31   136.2 1833.39   210.7 1791.71
   225.9 1781.65   232.3 1774.59   245.4 1742.19   250.1 1732.97     276  1715.3
   289.1 1704.43   302.2 1690.88     323 1672.85   335.1 1658.82     359 1636.44
   368.5 1632.77   383.7 1632.17   432.1 1633.53   447.1 1636.18   459.2    1640
   600.6 1638.44   663.8 1650.88   738.1 1655.26   777.8  1659.7   819.9 1670.94
#Mann= 7 ,-1 , 0
       0      .1       0    92.2      .1       0     359    .045       0
   447.1      .1       0  453.29      .1       0  566.86      .1       0
  803.54      .1       0
Bank Sta=359,447.1
XS Rating Curve= 0 ,0
Exp/Cntr=0.3,0.1

Type RM Length L Ch R = 1 ,7923    ,429.6,445.6,473.4
XS GIS Cut Line= 3
2425657.78284634674199.507475167     2425300.504      673998.484
     2424936.107      673812.895
#Sta/Elev= 30
       0 1734.98    21.8 1725.61    52.6 1714.96    90.8 1702.97   141.2 1689.76
   161.3 1682.63   177.9 1674.09   205.3 1651.33   221.5 1640.73   228.8 1637.68
   243.5 1635.82   311.2 1635.62   334.6 1633.94   352.3 1629.21     389 1629.43
   402.8 1628.12   438.9 1628.35   455.6 1630.93   467.5 1633.08   565.6 1632.41
   600.5 1634.68   622.9 1644.48   636.4 1652.29   649.8 1663.31   681.6 1683.47
   712.7 1696.48   761.9  1709.7   770.8 1715.48   782.7 1717.62   818.9 1733.59
#Mann= 4 ,-1 , 0
       0      .1       0     389    .045       0   455.6      .1       0
  654.06      .1       0
Bank Sta=389,455.6
XS Rating Curve= 0 ,0
Exp/Cntr=0.3,0.1

Type RM Length L Ch R = 1 ,7478    ,268.7,292,320.6
XS GIS Cut Line= 3
     2425722.476      674142.9592425704.85678492673962.968255423
2425400.91625299 673325.63698581
#Sta/Elev= 30
       0 1723.63    40.3 1699.94    60.4 1692.13    72.4 1690.06    92.5 1679.41
   136.7 1667.18   229.7 1650.52   266.5 1630.95   402.5 1628.78   429.1 1630.23
   522.2 1625.69   539.6 1622.98   570.9 1622.81   593.1 1625.65   601.9 1628.84
   610.8  1635.3   615.2 1642.06   624.1 1662.58   628.5 1669.05   641.1 1680.61
   662.6 1707.47   689.6 1730.06   721.6 1750.38     757 1765.52   805.8 1782.04
   819.1 1783.17   832.4 1790.14   845.5 1787.17   875.6 1787.06   886.9 1792.72
#Mann= 4 ,-1 , 0
       0      .1       0   522.2    .045       0   593.1      .1       0
  770.23     .06       0
Bank Sta=522.2,593.1
XS Rating Curve= 0 ,0
Exp/Cntr=0.3,0.1

Type RM Length L Ch R = 1 ,7186    ,320.4,312.4,293.4
XS GIS Cut Line= 3
2425763.47581087674150.323167849 2425718.5480969673906.062316846
2425960.83513237673301.488468072
#Sta/Elev= 30
       0 1737.24    48.2 1709.69    76.7 1696.62   105.2 1684.58   145.8 1671.19
   206.8 1657.15   273.3 1645.76     338 1629.36   350.9 1621.63   398.3 1624.32
   419.8 1619.33     454 1620.47   493.1 1619.66   509.4 1620.77   540.1  1623.5
   553.4 1628.93   566.4 1630.29   618.1 1625.21   661.2 1624.99   682.7 1619.81
   691.3 1619.06   708.6 1623.04   751.6 1624.11     756 1625.17   781.8 1639.62
     812 1652.93   829.2 1658.44   860.1 1658.75   876.6 1655.59   899.7 1656.24
#Mann= 5 ,-1 , 0
       0      .1       0     454    .045       0   509.4      .1       0
  615.08    .055       0  728.48      .1       0
#XS Ineff= 2 , 0
                          565.71         1638.18
Permanent Ineff=
       F       F
Bank Sta=454,509.4
XS Rating Curve= 0 ,0
Exp/Cntr=0.3,0.1

Type RM Length L Ch R = 1 ,6873    ,455.8,450,435.5
XS GIS Cut Line= 3
     2426103.268      674180.587     2426095.449      673771.906
2426095.52964806673259.211485485
#Sta/Elev= 30
       0 1861.42    73.7  1821.4    78.7 1817.87   109.7 1789.77   173.7 1753.14
   261.3 1698.29   317.8 1662.33   341.8 1646.06   357.8 1633.64   369.8 1621.71
   373.8 1619.39   381.8  1618.1   393.8 1615.46   453.8 1615.78   462.5 1617.41
   469.8 1622.21   485.8 1623.66   561.8  1623.2   597.8 1621.79   625.8 1622.65
   713.8 1621.44   733.8  1622.9   762.5 1623.33   777.8 1622.33   790.5 1616.75
   806.5 1616.26   814.5 1617.32   854.5  1632.5   909.8 1640.39   921.5 1641.21
#Mann= 5 ,-1 , 0
       0      .1       0   381.8    .045       0   462.5      .1       0
  652.38    .055       0  751.09      .1       0
Bank Sta=381.8,462.5
XS Rating Curve= 0 ,0
Exp/Cntr=0.3,0.1

Type RM Length L Ch R = 1 ,6423    ,473.9,450,430.3
XS GIS Cut Line= 3
     2426649.691      674090.553     2426537.942       673696.85
2426324.64526217673095.062786512
#Sta/Elev= 30
       0 1910.13    53.7 1890.36   132.7 1854.96   178.4 1830.32   215.9 1804.38
     258 1763.99   278.2 1741.99   282.4 1736.19   290.7 1717.45   294.9 1711.54
   328.1 1674.35     378 1631.99   382.2 1626.73   390.5 1611.27   394.7  1608.1
   406.3 1607.82   432.6 1608.05   442.8 1611.03   462.3 1617.45     492 1618.33
   801.8 1616.16   878.2 1618.54   895.1 1613.43   912.1 1613.57   929.1 1620.91
   941.8 1629.61   971.5  1654.3  1026.7 1652.48  1035.2 1655.05  1047.7 1663.05
#Mann= 6 ,-1 , 0
       0      .1       0   390.5    .045       0   442.8      .1       0
  449.37    .055       0  846.41      .1       0 1044.92     .06       0
Bank Sta=390.5,442.8
XS Rating Curve= 0 ,0
Exp/Cntr=0.3,0.1

Type RM Length L Ch R = 1 ,5973    ,442.8,450.5,467.6
XS GIS Cut Line= 3
     2427238.314      673643.571     2426888.577      673430.624
2426420.96735686673106.691837428
#Sta/Elev= 30
       0 1714.23    22.9 1701.12      37  1698.2    78.8 1709.71   130.6 1731.15
   177.5 1734.79     209 1729.24   238.9 1718.79   262.8 1704.54   285.4 1684.43
   302.9 1671.19   313.3 1660.55   324.3 1645.26   341.4 1631.31   355.1 1614.47
   364.8 1606.25   374.1 1603.05   416.3 1602.84   430.1 1603.98   436.5 1607.01
   445.8 1611.86   652.1 1613.31   781.4 1614.06   804.4  1610.2   825.3 1609.42
   856.2 1620.73   867.7 1628.51   887.8 1647.02   898.3 1653.19   978.3 1653.17
#Mann= 6 ,-1 , 0
       0      .1       0   364.8    .045       0   436.5      .1       0
  446.14    .055       0  641.45      .1       0  729.31    .055       0
Bank Sta=364.8,436.5
XS Rating Curve= 0 ,0
Exp/Cntr=0.3,0.1

Type RM Length L Ch R = 1 ,5523    ,441.8,454,475.6
XS GIS Cut Line= 3
     2427380.139      673440.671     2427164.653      673090.646
     2426936.314      672751.045
#Sta/Elev= 30
       0 1693.77    10.3 1689.51    56.1  1679.3   118.6 1652.19   141.9 1645.53
   193.4 1633.74   229.1 1631.49   265.1 1610.18   274.5 1601.83   300.2 1601.33
   310.5  1605.5   323.1  1607.1   354.4 1600.82     411 1601.24   464.6 1600.24
   472.8 1601.45   481.4 1604.68   501.6 1605.52   516.8 1609.78   572.2 1619.06
   603.5 1619.32   615.2 1624.95   656.6 1631.06   671.6 1638.82   691.8 1639.76
   709.6 1638.38   717.7 1640.89   743.7 1643.77   772.3 1650.15   820.3 1666.52
#Mann= 6 ,-1 , 0
       0      .1       0     411    .045       0   472.8      .1       0
  642.54    .055       0  653.28     .06       0  760.98      .1       0
Bank Sta=411,472.8
XS Rating Curve= 0 ,0
Exp/Cntr=0.3,0.1

Type RM Length L Ch R = 1 ,5069    ,307.9,300,298.3
XS GIS Cut Line= 3
      2427581.39      673378.019     2427591.489      672962.206
2427579.71869978 672520.32197162
#Sta/Elev= 30
       0 1674.12   131.2 1645.22   160.6 1633.68   191.9 1624.37   219.2 1618.59
   235.2 1617.29     252 1611.52   267.2 1602.38   275.2 1599.43   299.2 1594.49
   315.2 1594.15   347.2  1596.7   366.8 1597.04   387.2 1595.88   427.3 1594.79
   435.3 1596.09   443.2 1601.27   447.3 1602.63   467.9 1600.97   614.8 1599.84
   652.9  1603.1   711.4  1604.7   751.4 1604.35   783.4  1609.8   807.4 1611.02
   819.4 1610.33   843.4 1612.49   851.4 1614.75   855.4  1620.7     858  1627.6
#Mann= 5 ,-1 , 0
       0      .1       0   387.2    .045       0   435.3      .1       0
  476.91     .05       0  771.92     .06       0
Bank Sta=387.2,435.3
XS Rating Curve= 0 ,0
Exp/Cntr=0.3,0.1

Type RM Length L Ch R = 1 ,4769    ,450.7,440.6,435.5
XS GIS Cut Line= 3
     2427918.133      673432.021     2427881.413      673025.651
2427825.98194324672443.595207987
#Sta/Elev= 30
       0 1667.97    21.2 1661.12    49.3 1654.69   129.4 1642.14   274.2 1630.29
   278.3 1628.93   286.3 1621.19   302.5 1606.71   318.4 1598.83   362.6 1593.62
   374.7 1590.63   398.7 1590.47   425.9 1592.43   483.1 1593.49   503.2 1598.33
   515.3 1599.16   579.6 1597.45   756.4 1595.77   812.3 1599.54   844.8 1598.08
     870 1599.26   880.9 1599.95   893.6 1596.12   897.3 1596.59   913.1 1604.76
   957.3 1607.79   961.3 1609.57     967  1618.2     978 1642.51   992.7 1661.23
#Mann= 8 ,-1 , 0
       0      .1       0   129.4      .1       0   286.3      .1       0
   362.6    .045       0   425.9      .1       0   579.6     .05       0
     870    .055       0     967      .1       0
#XS Ineff= 2 , 0
                           876.9            1605
Permanent Ineff=
       F       F
Bank Sta=362.6,425.9
XS Rating Curve= 0 ,0
Exp/Cntr=0.3,0.1

Type RM Length L Ch R = 1 ,4328    ,474.4,459.4,446.7
XS GIS Cut Line= 2
2428416.97950245673245.0250446972428109.62301214672340.773341341
#Sta/Elev= 30
       0 1626.12    56.7 1621.42   107.9 1618.68   161.1 1612.97   171.2 1610.99
   188.1 1601.56   202.1 1598.28   209.3 1595.35   218.2 1594.73   233.6 1591.96
   276.9 1591.03   281.1 1590.13   289.5 1586.35   302.2 1585.14   314.9 1583.85
   361.4 1583.72     374 1585.36   424.7 1594.98   437.4 1591.61   471.2 1589.85
   576.8 1592.37   813.8 1591.55   857.5 1594.58     881 1594.08   889.5 1597.69
   902.1 1606.48   910.6 1614.15   923.2 1629.86   927.5  1634.3   955.1 1652.12
#Mann= 8 ,-1 , 0
       0     .05       0    77.7     .06       0  176.72      .1       0
   302.2    .045       0     374      .1       0   473.8     .05       0
  770.87     .06       0   869.9      .1       0
Bank Sta=302.2,374
XS Rating Curve= 0 ,0
Exp/Cntr(USF)=0,0
Exp/Cntr=0.3,0.1

Type RM Length L Ch R = 1 ,3869    ,316.3,334.9,351.2
XS GIS Cut Line= 3
2429055.51358869673112.913427935     2428686.658      672666.544
2428388.77598581672310.374125279
#Sta/Elev= 30
       0 1628.56    32.6 1619.92    45.2 1615.03    53.1 1610.19    70.1 1606.33
   109.9  1589.3   142.7  1583.6   376.2 1585.93   495.6 1584.52   516.1 1588.53
   527.6 1587.46     535 1584.01   541.2 1580.41   547.2 1578.74   564.5 1578.45
     610 1578.84   630.7 1582.94   649.7 1590.32     660 1586.28   667.2 1585.36
     752  1586.1   811.6 1588.74   870.6 1588.27   980.1 1589.69   985.3 1591.29
     999  1602.4  1015.4 1620.13  1021.8 1629.24  1027.4 1635.58  1043.4 1648.03
#Mann= 9 ,-1 , 0
       0      .1       0   51.22     .05       0  391.66     .06       0
  505.14    .055       0     535    .045       0   630.7     .05       0
  732.64     .06       0  926.32    .035       0   960.4     .06       0
Bank Sta=535,630.7
XS Rating Curve= 0 ,0
Exp/Cntr=0.3,0.1

Type RM Length L Ch R = 1 ,3534    ,89,85.2,88
XS GIS Cut Line= 2
2429121.94140326673099.6454121762428829.47287317672175.119892069
#Sta/Elev= 30
       0 1621.38    34.4 1619.75    93.1 1610.33   130.8 1598.76   139.2 1594.19
   151.8 1585.19   164.4 1580.52   181.6 1580.19   227.3 1582.49   420.7 1584.45
   588.1 1580.85   663.7 1582.41   671.3 1578.58   676.2 1575.35   680.4 1574.67
     714 1573.72     756 1574.15   760.2 1574.98   766.5 1578.63   774.4 1581.82
   802.1 1584.24   827.3 1593.26   866.9 1594.07   877.6 1600.21   890.2 1610.33
   902.8 1622.68     907    1625   923.8 1632.83   936.4 1634.63   969.7 1647.15
#Mann= 9 ,-1 , 0
       0      .1       0  140.27     .05       0  436.31     .06       0
  534.99    .035       0  633.67    .055       0   671.3    .045       0
   766.5    .055       0  831.03     .06       0  929.71      .1       0
Bank Sta=671.3,766.5
XS Rating Curve= 0 ,0
Exp/Cntr(USF)=0,0
Exp/Cntr=0.5,0.3

Type RM Length L Ch R = 1 ,3449    ,37,36.6,37.8
XS GIS Cut Line= 3
2429168.54588077673135.0320051772428987.04515263672391.167316155
2428917.53040144672116.519073846
#Sta/Elev= 30
       0 1634.56    37.2 1618.86      66 1619.57   111.3 1613.36   173.1 1598.12
   197.8 1585.25   210.1 1584.25   226.6 1579.75   255.4 1582.49   399.5 1581.84
   518.9 1583.65   683.6 1578.94   736.4 1581.25   745.4 1579.61   749.3 1576.67
   757.7 1571.63   778.4 1571.04   807.2 1571.46   811.4 1573.43   815.4 1578.02
   823.7    1586   836.1 1592.97   873.3 1596.42   902.1 1596.65   914.5 1605.38
   939.3  1607.9   955.8 1621.13  1026.3 1636.88  1042.4 1645.71    1049 1647.18
#Mann= 8 ,-1 , 0
       0      .1       0  181.43     .05       0     573     .06       0
   670.9    .055       0   749.3    .045       0   815.4     .06       0
  964.73      .1       0 1010.26      .1       0
#XS Ineff= 2 , 0
             740    1580     819            1582
Permanent Ineff=
       F       F
Bank Sta=749.3,815.4
XS Rating Curve= 0 ,0
Exp/Cntr=0.5,0.3

Type RM Length L Ch R = 1 ,3412    ,108.1,109.2,110.8
XS GIS Cut Line= 2
2429190.18406028673122.3929645162428964.33336204672126.375137054
#Sta/Elev= 30
       0 1628.57    29.2 1615.84    81.5 1613.45     102 1610.31   151.2 1597.78
   175.9 1588.97   188.2 1587.43   208.7 1579.91   245.6  1582.2   339.6 1581.28
   524.5 1583.04   684.5 1578.37   700.9 1579.26   717.3 1582.61   733.7  1576.5
     748 1570.72   770.6 1570.31   791.1 1571.68   804.9 1577.73   814.9 1588.27
   823.9 1591.76   860.8 1597.07   889.5 1597.24   905.9 1608.04     910 1609.32
   930.5 1609.23     951 1612.53   978.7 1621.28  1004.4 1626.33  1021.3 1633.88
#Mann= 8 ,-1 , 0
       0     .05       0   87.94      .1       0  172.01     .05       0
  563.09     .06       0  660.86    .055       0   733.7    .045       0
   804.9     .06       0  954.17      .1       0
Bank Sta=733.7,804.9
XS Rating Curve= 0 ,0
Exp/Cntr(USF)=0,0
Exp/Cntr=0.5,0.3

Type RM Length L Ch R = 1 ,3303    ,328.1,334.1,340.3
XS GIS Cut Line= 2
2429264.92601797673107.7695380122429084.57042441672116.626186052
#Sta/Elev= 30
       0 1615.02    13.1  1608.9    19.8 1607.18    37.5 1606.27    85.2 1599.54
   118.8 1596.57   126.9 1594.27   146.2 1584.27   167.4  1579.2   253.7 1582.42
   302.6 1580.27   468.4 1581.13   589.8 1579.13   631.1 1580.15   704.3 1576.72
   716.5 1579.35     724 1575.61   735.3 1570.31   765.2 1569.83   793.8 1571.51
   801.8 1573.58   805.9 1576.11   818.4 1589.64   826.2 1594.71   852.3  1596.5
   883.6 1597.37   895.3 1601.67     936 1606.56   950.6 1610.38  1007.4  1632.6
#Mann= 5 ,-1 , 0
       0     .05       0     724    .045       0   805.9      .1       0
   852.3    .055       0   950.6      .1       0
#XS Ineff= 2 , 0
           253.7    1595
Permanent Ineff=
       F       F
Bank Sta=724,805.9
XS Rating Curve= 0 ,0
Exp/Cntr(USF)=0,0
Exp/Cntr=0.3,0.1

Type RM Length L Ch R = 1 ,2969    ,451.1,450,450.1
XS GIS Cut Line= 3
     2429499.326 673114.96633014      2429454.92      672288.874
2429434.18773052671971.744375962
#Sta/Elev= 30
       0 1604.81    40.1 1597.88    56.2 1594.07    68.2 1589.65    80.2 1579.11
    88.4  1576.4   124.3 1575.86   176.3 1577.45   256.4 1576.63     453 1577.48
   580.9 1575.81     633 1572.28   697.1 1572.27   713.1 1574.14   777.2 1574.43
   781.2 1573.52   797.2 1567.38   853.3 1566.81   869.4 1568.69   873.4 1570.11
   878.2 1573.93   889.4 1584.34   893.4 1586.72   897.4 1587.63   929.5 1589.45
   937.5  1593.2   953.6 1594.07  1041.7  1604.6  1117.9 1623.18  1145.1 1628.82
#Mann= 7 ,-1 , 0
       0      .1       0  114.77     .06       0   506.9      .1       0
   781.2    .045       0   878.2     .06       0  898.95    .055       0
  996.87     .05       0
Bank Sta=781.2,878.2
XS Rating Curve= 0 ,0
Exp/Cntr=0.3,0.1

Type RM Length L Ch R = 1 ,2519    ,490.4,493.4,498.2
XS GIS Cut Line= 3
2429978.75546103673294.663716807     2429901.246      672299.192
     2429871.081      671890.805
#Sta/Elev= 30
       0 1650.91    51.9 1617.76      84 1602.05   104.1 1595.19   180.3 1585.63
   184.3 1581.97   192.4 1570.44   196.4 1568.84   284.6 1570.48   320.7 1569.04
   413.1 1571.69   477.2 1569.45   557.5 1569.71   625.7 1566.66   709.9 1570.27
   762.1 1570.18   806.2 1563.46   918.5 1569.41   938.6 1569.03   945.3  1566.1
   956.4 1560.78   990.8 1560.42  1014.8 1560.82  1038.9 1565.26    1063 1579.59
    1095 1578.12  1111.1 1581.81  1327.7 1588.05  1391.9 1592.11    1408 1595.05
#Mann= 9 ,-1 , 0
       0      .1       0  268.61     .05       0  464.26    .055       0
  562.09     .06       0  659.91     .05       0   945.3    .045       0
  1038.9     .05       0 1051.22    .055       0 1149.08     .05       0
Bank Sta=945.3,1038.9
XS Rating Curve= 0 ,0
Exp/Cntr=0.3,0.1
